--- MinearRun.prj (project) ---

Proj Title=MinearRun
Current Plan=p01
Default Exp/Contr=0.3,0.1
SI Units
Geom File=g01
Flow File=f01
Plan File=p01
Background Map Layer=Bing Satellite
Y Axis Title=Elevation
X Axis Title(PF)=Main Channel Distance
X Axis Title(XS)=Station
BEGIN DESCRIPTION:
September 2018
Tucker County ABFE Study
US Army Corps of Engineers, Pittsburgh District
NAD 1983 UTM 17N (meters)
END DESCRIPTION:
DSS Export Rating Curves= 0
DSS Export Rating Curve Sorted= 0
DSS Export Volume Flow Curves= 0
DXF OffsetX= 0
DXF OffsetY= 0
DXF ScaleX= 1
DXF ScaleY= 10

--- MinearRun.p01 (plan) ---

Plan Title=MinearRun_plan
Program Version=5.05
Short Identifier=Plan1_subcritical
Geom File=g01
Flow File=f01
Subcritical Flow
K Sum by GR= 0
Std Step Tol= 0.003
Critical Tol= 0.003
Num of Std Step Trials= 20
Max Error Tol= 0.1
Flow Tol Ratio= 0.001
Split Flow NTrial= 30
Split Flow Tol= 0.006
Split Flow Ratio= 0.02
Log Output Level= 0
Friction Slope Method= 1
Unsteady Friction Slope Method= 2
Unsteady Bridges Friction Slope Method= 1
Parabolic Critical Depth
Global Vel Dist= 0 , 0 , 0
Global Log Level= 0
CheckData=True
Encroach Param=-1 ,0,0, 0
Computation Interval=1MIN
Output Interval=1HOUR
Instantaneous Interval=1HOUR
Mapping Interval=1HOUR
Computation Time Step Use Courant=        0
Computation Time Step Use Time Series=    0
Computation Time Step Count To Double=0
Computation Time Step Max Doubling=0
Computation Time Step Max Halving=0
Computation Time Step Residence Courant=0
Run HTab= 0
Run UNet= 0
Run Sediment= 0
Run PostProcess= 0
Run WQNet= 0
Run RASMapper=-1
UNET Theta= 1
UNET Theta Warmup= 1
UNET ZTol= 0.006
UNET ZSATol= 0.006
UNET MxIter= 20
UNET Max Iter WO Improvement= 0
UNET MaxInSteps= 0
UNET DtIC= 0
UNET DtMin= 0
UNET MaxCRTS= 20
UNET WFStab= 2
UNET SFStab= 1
UNET WFX= 1
UNET SFX= 1
UNET 1D Methodology=Finite Difference
UNET DSS MLevel= 4
UNET Pardiso=0
UNET DZMax Abort= 30
UNET Use Existing IB Tables=-1
UNET Froude Reduction=False
UNET Froude Limit= 0.8
UNET Froude Power= 4
UNET D1 Cores= 0
UNET D2 Coriolis=0
UNET D2 Cores= 0
UNET D2 Theta= 1
UNET D2 Theta Warmup= 1
UNET D2 Z Tol= 0.003
UNET D2 Volume Tol= 0.003
UNET D2 Max Iterations= 20
UNET D2 Equation= 0
UNET D2 RampUpFraction=0.1
UNET D2 TimeSlices= 1
UNET D2 BCVolumeCheck=0
UNET D1D2 MaxIter= 0
UNET D1D2 ZTol=0.003
UNET D1D2 QTol=0.1
UNET D1D2 MinQTol=0.03
Write IC File= 0
Write IC File at Fixed DateTime=0
Write IC File at Sim End=0
Echo Input=False
Echo Parameters=False
Echo Output=False
Write Detailed= 0
HDF Write Warmup=0
HDF Write Time Slices=0
HDF Flush=0
HDF Face Node Velocities=0
HDF Compression= 1
HDF Chunk Size= 1
HDF Spatial Parts= 1
HDF Use Max Rows=0
HDF Fixed Rows= 1
Calibration Method= 0
Calibration Iterations= 20
Calibration Max Change=0.05
Calibration Tolerance=0.2
Calibration Maximum=1.5
Calibration Minimum=0.5
Calibration Optimization Method= 1
WQ AD Non Conservative
WQ ULTIMATE=-1
WQ Max Comp Step=1HOUR
WQ Output Interval=15MIN
WQ Output Selected Increments= 0
WQ Output face flow=0
WQ Output face velocity=0
WQ Output face area=0
WQ Output face dispersion=0
WQ Output cell volume=0
WQ Output cell surface area=0
WQ Output cell continuity=0
WQ Output cumulative cell continuity=0
WQ Output face conc=0
WQ Output face dconc_dx=0
WQ Output face courant=0
WQ Output face peclet=0
WQ Output face adv mass=0
WQ Output face disp mass=0
WQ Output cell mass=0
WQ Output cell source sink temp=0
WQ Output nsm pathways=0
WQ Output nsm derived pathways=0
WQ Output MaxMinRange=-1
WQ Daily Max Min Mean=-1
WQ Daily Range=0
WQ Daily Time=0
WQ Create Restart=0
WQ Fixed Restart=0
WQ System Summary=0
WQ Write To DSS=0
WQ Use Fixed Temperature=0
Sorting and Armoring Iterations= 10
XS Update Threshold= 0.02
Bed Roughness Predictor= 0
Hydraulics Update Threshold= 0.02
Energy Slope Method= 1
Volume Change Method= 1
Sediment Retention Method= 0
XS Weighting Method= 0
Number of US Weighted Cross Sections= 1
Number of DS Weighted Cross Sections= 1
Upstream XS Weight=0
Main XS Weight=1
Downstream XS Weight=0
Number of DS XS's Weighted with US Boundary= 1
Upstream Boundary Weight= 1
Weight of XSs Associated with US Boundary= 0
Number of US XS's Weighted with DS Boundary= 1
Downstream Boundary Weight= 0.5
Weight of XSs Associated with DS Boundary= 0.5
Percentile Method= 0
Sediment Output Level= 4
Mass or Volume Output= 0
Output Increment Type= 1
Profile and TS Output Increment= 1
XS Output Flag= 0
XS Output Increment= 10
Write Gradation File= 0
Read Gradation Hotstart= 0
Write HDF5 File= 1
Write Binary Output= 1
Write DSS Sediment File= 0
SV Curve= 0
Specific Gage Flag= 0

--- MinearRun.f01 (steady flow) ---

Flow Title=MinearRun_flow
Program Version=5.05
Number of Profiles= 1
Profile Names=PF 1
River Rch & RM=Little Mill Run,1               ,365.7599
  9.4323
River Rch & RM=Little Mill Run,1               ,91.62041
  9.7409
River Rch & RM=Mill Run(Minear),2               ,3200.4
   14.64
River Rch & RM=Mill Run(Minear),2               ,2286
 16.1121
River Rch & RM=Mill Run(Minear),2               ,1591.275
 17.7262
River Rch & RM=Mill Run(Minear),2               ,1491.988
 19.5384
River Rch & RM=Mill Run(Minear),2               ,731.52
 21.4923
River Rch & RM=Mill Run(Minear),2               ,365.76
 28.0051
River Rch & RM=Mill Run(Minear),1               ,274.2707
   28.26
River Rch & RM=Mill Run(Minear),1               ,19.92903
 28.3732
River Rch & RM=Minear Run,1               ,7376.625
  40.681
River Rch & RM=Minear Run,1               ,6492.24
 41.7386
River Rch & RM=Minear Run,1               ,5303.417
 45.8729
River Rch & RM=Minear Run,1               ,4297.68
 47.7984
River Rch & RM=Minear Run,1               ,4206.24
  53.363
River Rch & RM=Minear Run,1               ,3108.96
 54.8209
River Rch & RM=Minear Run,1               ,692.6317
 60.8806
River Rch & RM=Stump Run,1               ,1828.007
   14.64
River Rch & RM=Stump Run,1               ,1188.022
  16.282
River Rch & RM=Stump Run,1               ,90.74239
 17.9244
River Rch & RM=Stump Run,1               ,2.381145
 17.9527
Boundary for River Rch & Prof#=Little Mill Run,1               , 1
Up Type= 2
Dn Type= 0
Boundary for River Rch & Prof#=Mill Run(Minear),2               , 1
Up Type= 2
Dn Type= 0
Boundary for River Rch & Prof#=Mill Run(Minear),1               , 1
Up Type= 0
Dn Type= 0
Boundary for River Rch & Prof#=Minear Run,1               , 1
Up Type= 0
Dn Type= 1
Dn Known WS=473.2
Boundary for River Rch & Prof#=Stump Run,1               , 1
Up Type= 2
Dn Type= 0
DSS Import GetInterval= 0
DSS Import GetPeak= 0
DSS Import FillOption= 0

--- MinearRun.g01 (geometry) ---

Geom Title=MinearRun_geometry
Program Version=5.05

Junct Name=2
Junct Desc=, 0 , 0 , 0 ,0
Up River,Reach=Little Mill Run ,1
Up River,Reach=Mill Run(Minear),2
Dn River,Reach=Mill Run(Minear),1
Junc L&A=110,
Junc L&A=92,

Junct Name=4
Junct Desc=, 0 , 0 , 0 ,0
Up River,Reach=Mill Run(Minear),1
Up River,Reach=Stump Run       ,1
Dn River,Reach=Minear Run      ,1
Junc L&A=48,
Junc L&A=30,

River Reach=Little Mill Run ,1
Reach XY= 30
     615383.4468    4340557.6386     615372.3886    4340562.6283
     615366.8594    4340565.1231     615364.0949    4340566.3706
     615358.5657    4340568.8654     615350.2721    4340572.6077
     615344.7429    4340575.1025     615341.9784      4340576.35
     615336.4492    4340578.8448      615325.391    4340583.8345
     615303.0682    4340590.9977     615300.2779    4340591.8932
     615277.9551    4340599.0564      615232.603    4340578.3085
     615222.1239    4340567.1335     615213.7405    4340558.1936
     615203.2614    4340547.0186     615187.0864    4340538.5226
     615184.3905    4340537.1067     615168.2155    4340528.6107
     615131.2567    4340502.7564     615126.6454    4340498.7498
     615124.3397    4340496.7466     615117.4228    4340490.7367
     615112.8114    4340486.7302     615105.8945    4340480.7203
     615103.5888    4340478.7171     615098.9775    4340474.7105
     615090.5108    4340465.8911     615073.5775    4340448.2522

Type RM Length L Ch R = 1 ,365.7599,90.48,91.44,93.1
XS GIS Cut Line= 3
     615368.2423    4340535.2412     615386.2331    4340575.1126
     615408.7141    4340647.6346
#Sta/Elev= 20
       0  583.27    2.92  580.59    5.83  577.76    8.75  575.41   11.66  574.09
   14.58  573.53   18.88 573.064   23.33  572.62   50.02573.0646   61.96  573.26
   71.08  573.57   83.22  574.38   86.26  574.54    89.3  574.59   95.37  575.05
   98.41   575.8  101.45  577.17  113.59  583.26  116.63  583.68  119.67  584.87
#Mann= 3 , 0 , 0
       0      .1       0   18.88      .1       0   50.02      .1       0
Bank Sta=18.88,50.02
XS Rating Curve= 0 ,0
Exp/Cntr=0.3,0.1

Type RM Length L Ch R = 1 ,274.3199,79.6,91.44,105.01
XS GIS Cut Line= 2
     615278.4718    4340543.6429     615317.3164     4340664.694
#Sta/Elev= 24
       0   586.3    3.03  583.93    9.08  578.03   12.11  575.23   15.13  572.85
   18.16  571.34   21.19  570.84   23.25570.7993   42.38  570.58   57.51  570.52
   60.54  570.55   63.72570.7994   69.62   571.5    78.7  572.22   81.73  572.61
   84.75   573.3   87.78  574.18   90.81   574.2  105.94     579     112  581.13
  115.02  582.31  118.05  583.02  121.08  583.52  127.13   586.4
#Mann= 3 , 0 , 0
       0      .1       0   23.25      .1       0   63.72      .1       0
Bank Sta=23.25,63.72
XS Rating Curve= 0 ,0
Exp/Cntr=0.3,0.1

Type RM Length L Ch R = 1 ,182.88  ,91.87,91.26,68.32
XS GIS Cut Line= 5
     615240.2211    4340533.7266     615218.7468    4340558.2034
     615205.9208    4340570.2309     615186.3121    4340602.5184
     615245.0242    4340670.6609
#Sta/Elev= 30
       0  587.65   17.76  572.21   20.72   571.4   23.68  570.26   26.64  569.35
   32.56  568.96   35.26568.6833   38.42  568.41   44.28  568.21   50.14  568.37
   54.15568.6832   61.77  569.08    79.2   569.6   87.92  569.48   99.91   570.1
  111.91  570.17   117.9  570.03   120.9  570.17   126.9  571.06  135.89  572.71
  138.89  572.81  141.89  573.19  147.89  574.41  150.88  575.14  153.88  576.19
  159.88  579.06  168.87  583.69  171.87  584.03  174.87     585  177.87  586.76
#Mann= 3 , 0 , 0
       0      .1       0   35.26      .1       0   54.15      .1       0
Bank Sta=35.26,54.15
XS Rating Curve= 0 ,0
Exp/Cntr=0.3,0.1

Type RM Length L Ch R = 1 ,91.62041,86.59,91.62,15.07
XS GIS Cut Line= 5
     615173.0549    4340465.4925     615133.1301    4340521.0163
     615142.6888    4340541.0688     615134.0899    4340558.9283
     615236.9858    4340670.4119
#Sta/Elev= 30
       0  585.69    2.97     585    5.95  583.84    8.92  582.06   11.89  580.81
   17.84  577.53   20.81  576.23   38.65  569.49    44.6  568.18   47.57  567.11
   52.64566.5518   73.94  566.07   82.07 566.552    90.6  567.36   96.27  567.61
  110.42  567.45  140.77  568.25  162.01  568.02  192.35  570.09  207.52  570.72
  210.55  571.01  216.62  571.75  219.66  572.33  225.72   572.9  237.86  575.38
   240.9  576.27  243.93  577.66     250  581.09  256.07  584.19  262.13  585.53
#Mann= 3 , 0 , 0
       0      .1       0   52.64      .1       0   82.07      .1       0
Bank Sta=52.64,82.07
XS Rating Curve= 0 ,0
Exp/Cntr=0.3,0.1

River Reach=Mill Run(Minear),2
Reach XY= 30
     616689.1265    4342482.9021     616664.7848    4342388.7102
616619.345170091 4342335.8059044616529.8147348624342273.50871633
      616501.272    4342229.9599 616495.638948994342172.54323009
     616457.88024342156.25329303     616434.5968    4342111.9555
616394.4944629354342087.41196037     616390.6759    4342035.2262
     616290.1341    4341953.2052     616214.4631    4341862.7175
616168.726504953 4341766.3325811616152.8301306414341748.39972294
     615987.4501    4341708.7297     615906.4875    4341648.9337
     615859.3509     4341592.557615867.2941212834341521.44045321
615796.6892398164341448.37717633615672.5595908254341417.37586018
615553.9759976154341438.10676294     615409.8472    4341346.8134
      615261.432    4341306.5622     615218.0402    4341263.1705
     615159.3026    4341166.2666     615115.9109    4340985.8866
     615107.5376     4340888.831 615132.622948994340819.43842569
     615085.7483    4340613.8817     615073.5775    4340448.2522

Type RM Length L Ch R = 1 ,3200.4  ,95.36,91.44,67.13
XS GIS Cut Line= 4
     616730.5228    4342451.6801     616672.3172    4342453.1172
     616641.7888    4342463.1383     616599.6644     4342487.048
#Sta/Elev= 28
       0  648.61    3.06  647.17    6.13  646.33   21.45  642.93   24.52  641.93
   27.58  641.15   30.64  640.16   33.71  638.98   34.72638.7258   36.77  638.21
   39.84  638.04   59.49638.7265   66.99  639.17   75.75  639.45   81.59   639.8
   84.51  639.79   87.43  639.63   90.35  639.29   93.38  639.09   99.44  639.64
  102.46  639.66  111.55  639.06  114.57  639.08   117.6  639.59  120.63  640.46
  132.74  644.44  135.76   646.1  138.79  647.41
#Mann= 3 , 0 , 0
       0      .1       0   34.72      .1       0   59.49      .1       0
Bank Sta=34.72,59.49
XS Rating Curve= 0 ,0
Exp/Cntr=0.3,0.1

Type RM Length L Ch R = 1 ,3108.96 ,22.3,20.8,19.58
XS GIS Cut Line= 4
     616665.5313    4342348.8559     616635.0209    4342392.3102
     616604.6387    4342425.4935     616573.8088    4342451.9191
#Sta/Elev= 29
       0  647.18     5.9  645.89    8.85  645.04   14.75  641.84    17.7  640.66
   20.65  639.51   26.55  637.78    29.5  636.74   31.45636.1785   32.45  635.89
    35.4  635.51   38.35  635.67   43.38636.1786   50.15  636.76    56.1  637.16
   65.09  637.38   83.09  637.49   95.09  637.31   98.09  637.23  103.89  636.68
  106.79  636.66  112.59  636.97  115.49  637.22  121.29  638.56  124.19  639.39
  127.09  640.56  129.99  642.18  135.79  645.89  138.69  647.58
#Mann= 3 , 0 , 0
       0      .1       0   31.45      .1       0   43.38      .1       0
Bank Sta=31.45,43.38
XS Rating Curve= 0 ,0
Exp/Cntr=0.3,0.1

Type RM Length L Ch R = 1 ,3088.156,27.01,26.59,20.46
XS GIS Cut Line= 6
     616657.0669    4342315.3245      616634.908    4342353.3584
     616628.9769    4342362.4821     616626.7941    4342371.6764
     616609.0008    4342392.1155     616559.3031    4342438.0649
#Sta/Elev= 30
       0  647.22    5.87   644.6   14.67  640.26   17.61  639.25   20.54   638.8
   23.48  639.03   26.41  639.11   29.35  638.87   35.21  637.23   38.15  636.75
   44.02  636.09   49.58635.7116    54.9   635.3   59.63   635.1   64.35  635.27
   67.36  635.59   69.52 635.712   82.42  636.87   88.44  637.14   91.45  637.12
  120.88  636.22  126.76   636.3  129.71  636.57  132.65  637.01  138.53  637.98
  141.48  639.49  144.42  640.85  147.36  643.23  153.25  646.57  159.13  649.67
#Mann= 3 , 0 , 0
       0      .1       0   49.58      .1       0   69.52      .1       0
Bank Sta=49.58,69.52
XS Rating Curve= 0 ,0
Exp/Cntr=0.3,0.1

Type RM Length L Ch R = 1 ,3061.569,24.51,24.75,27.99
XS GIS Cut Line= 5
     616641.0595    4342299.1584     616603.6209    4342352.0752
     616601.2397     4342366.495     616592.5084     4342384.619
     616547.1323    4342424.5711
#Sta/Elev= 30
       0  648.06   14.73  640.03   20.63  638.48   23.57  637.43   33.37 634.571
   35.36  633.91    38.3  633.84   41.25  634.31   44.75634.5718   50.09  634.93
   55.98  634.79   67.74  635.33   73.59  634.74   76.51  634.78   85.18  636.32
   90.93  637.08   99.55  637.46   105.6  637.38  108.62  637.07  114.67  636.04
  117.69  636.02  123.74  636.56  132.81  637.14  135.83  637.81  138.85  638.99
  141.87  639.83   144.9  641.08  150.94  643.99  156.99  647.85  160.01  649.25
#Mann= 3 , 0 , 0
       0      .1       0   33.37      .1       0   44.75      .1       0
Bank Sta=33.37,44.75
XS Rating Curve= 0 ,0
Exp/Cntr=0.3,0.1

Type RM Length L Ch R = 1 ,3036.819,15.64,19.3,18.67
XS GIS Cut Line= 6
     616633.9158    4342291.3532     616610.6324    4342310.6678
     616589.7303    4342322.3095     616581.3959    4342344.5345
     616576.5011    4342360.0127     616525.3041    4342407.6378
#Sta/Elev= 28
       0  648.63    9.08  643.89    12.1  641.54   15.13  639.65   21.18  636.64
    24.2  635.49   27.23  634.77   36.23  633.52   38.69 632.903   39.22  632.77
   42.21  632.52   45.21  632.51   55.78632.9019   71.98  633.98   80.62  634.02
   86.03  634.26   91.44  634.79   100.2  635.48  109.28  635.92  121.44  636.29
  124.48   636.7  130.57   639.3  133.62  640.85  136.66  642.17   145.8  645.17
  148.85  646.47  151.89  647.63  164.07  652.14
#Mann= 3 , 0 , 0
       0      .1       0   38.69      .1       0   55.78      .1       0
Bank Sta=38.69,55.78
XS Rating Curve= 0 ,0
Exp/Cntr=0.3,0.1

Type RM Length L Ch R = 1 ,3017.52 ,85.98,91.44,84.82
XS GIS Cut Line= 6
     616629.8844    4342278.1644     616585.4343    4342306.7395
       616564.38    4342339.6082     616557.6643    4342352.1118
      616548.276    4342363.2623     616519.2884    4342387.7021
#Sta/Elev= 30
       0  650.84    2.94  648.47    5.87  646.81    8.81  645.94   11.74  644.73
   14.68  642.88   17.61  641.58   26.42  636.45   29.36  634.52   37.83632.7421
    41.1  632.27   44.04  632.16   55.85   632.4   65.42632.7413   70.86  632.82
   85.87  633.37   94.71  633.46   97.58  633.64  106.07  634.86  108.98  634.88
  123.56  635.64  126.48  635.92   129.4  636.95  132.31   638.6  135.23   640.1
  138.15  641.86  141.06  643.17   146.9  645.11  155.64  647.76  158.56  648.12
#Mann= 3 , 0 , 0
       0      .1       0   37.83      .1       0   65.42      .1       0
Bank Sta=37.83,65.42
XS Rating Curve= 0 ,0
Exp/Cntr=0.3,0.1

Type RM Length L Ch R = 1 ,2926.08 ,79.97,91.44,92.65
XS GIS Cut Line= 6
     616579.5978    4342226.6504      616550.377     4342248.079
     616540.6111    4342264.1682     616537.7176    4342275.2158
     616530.2686    4342287.7666      616492.603    4342310.2594
#Sta/Elev= 27
       0  638.69    3.02  637.16    6.04  636.15    9.06  634.53   12.08  633.24
    15.1  632.57   18.12  632.13   21.14     632   33.22  631.76   36.24   631.6
   49.68  631.53   52.16631.4378   57.91  631.26   60.77  631.09   66.48  631.24
   75.23  630.91   78.15  630.87   81.07  631.04   83.98631.4373   86.92  632.04
   98.62  633.54  101.55  633.84  104.47  634.26  107.39  634.87  113.24  636.62
  119.09  637.77  124.94  639.05
#Mann= 3 , 0 , 0
       0      .1       0   52.16      .1       0   83.98      .1       0
Bank Sta=52.16,83.98
XS Rating Curve= 0 ,0
Exp/Cntr=0.3,0.1

Type RM Length L Ch R = 1 ,2834.64 ,37.58,37.25,35.42
XS GIS Cut Line= 4
     616546.8956     4342147.311     616497.6551    4342194.7104
     616487.4705     4342201.585     616460.7952    4342216.7664
#Sta/Elev= 24
       0  639.94    2.97  638.82    5.94  637.33    8.91  635.49   17.83  632.04
    20.8  631.24   29.72  629.61   32.69  629.24   38.63  628.57   47.55  628.16
   52.25627.6786   56.46  627.26   59.43  627.26   65.38  627.59   68.59 627.679
   71.42  628.02   80.63  628.73   89.84  629.74   92.91   630.5   95.98  633.18
   99.05   635.7  102.12  636.94  105.19  637.76  111.33     639
#Mann= 3 , 0 , 0
       0      .1       0   52.25      .1       0   68.59      .1       0
Bank Sta=52.25,68.59
XS Rating Curve= 0 ,0
Exp/Cntr=0.3,0.1

Type RM Length L Ch R = 1 ,2797.389,35.87,37.66,38.57
XS GIS Cut Line= 5
     616542.0611    4342125.0622     616507.6652    4342133.7935
      616483.588    4342156.5477     616462.4743    4342176.9206
     616436.1217    4342200.2569
#Sta/Elev= 30
       0  639.55   11.83  634.67   17.74  632.42    20.7  630.87   23.66  630.18
   26.62  629.66   35.49  628.56    38.5   628.1   44.52  627.48   48.98626.6313
   50.54  626.31   53.56  626.02   59.58  626.14    65.6  626.52   74.48  626.87
   77.42  626.83   83.28   626.5   86.59626.6317   92.09  627.38  100.89  628.16
  103.82  628.95  106.75  630.53  109.69  632.55  112.62  634.14  115.56  635.05
  118.49  636.68  121.42  638.12  124.35  639.14  130.22  640.95  133.15  642.01
#Mann= 3 , 0 , 0
       0      .1       0   48.98      .1       0   86.59      .1       0
Bank Sta=48.98,86.59
XS Rating Curve= 0 ,0
Exp/Cntr=0.3,0.1

Type RM Length L Ch R = 1 ,2759.728,14.97,16.53,17.53
XS GIS Cut Line= 5
     616535.0231    4342100.2442     616498.5106     4342114.373
     616471.9993    4342122.9455     616436.3598    4342147.5122
     616407.2291    4342168.2291
#Sta/Elev= 30
       0  638.17   12.05  634.18   24.09  631.59    27.1  630.83   30.12  629.73
   33.13  628.44   36.14  628.05   41.94  627.73   47.51   627.2    50.3  626.77
   53.58625.7693   55.87   625.4   58.65  625.23   64.23   625.3   72.79  625.81
    90.1   626.3   92.99  626.21   98.76  625.61    99.7625.7699  104.53  626.76
  107.41     627  113.28  626.98  116.26   627.3  119.24   628.3  125.19  631.27
  128.17   633.2  134.13  635.21  137.11   636.8  140.09  637.68  146.05  640.34
#Mann= 3 , 0 , 0
       0      .1       0   53.58      .1       0    99.7      .1       0
Bank Sta=53.58,99.7
XS Rating Curve= 0 ,0
Exp/Cntr=0.3,0.1

Type RM Length L Ch R = 1 ,2743.2  ,68.06,91.44,88.43
XS GIS Cut Line= 4
      616523.083    4342075.3442     616446.3258    4342122.2157
     616435.9115    4342126.8102     616397.9044    4342149.2522
#Sta/Elev= 30
       0  639.21       3  637.96   11.99  635.22   20.99  632.15   26.98  630.81
   29.98  629.77   35.97  628.59   38.97  627.61   41.97  626.99   57.52 625.584
   62.96  625.05   65.95  625.07   71.95  625.59   80.94   625.7   86.94  625.68
   89.94  625.56   95.63  625.05   98.47  625.08  101.72625.5839  104.26  626.18
   107.2  626.68  110.15  627.01  113.09  627.12  118.97  626.93  121.92   627.3
  124.86  628.39  136.63  633.59  139.57  635.67  142.52  637.22  145.46  638.55
#Mann= 3 , 0 , 0
       0      .1       0   57.52      .1       0  101.72      .1       0
Bank Sta=57.52,101.72
XS Rating Curve= 0 ,0
Exp/Cntr=0.3,0.1

Type RM Length L Ch R = 1 ,2651.76 ,93.46,91.44,76.63
XS GIS Cut Line= 6
     616485.8429    4342029.7696     616410.3962    4342077.9301
     616390.8263    4342077.3519     616383.9301    4342075.5047
     616377.0663    4342075.2868     616340.5553    4342079.4686
#Sta/Elev= 30
       0  638.16    2.98  636.74    5.97  635.67   11.93  634.73   14.92  635.41
    17.9  635.67   20.89  635.83   23.87  635.65   26.85  634.88   32.82  632.16
    35.8  630.64   41.77  626.68   44.75  625.75    53.7  624.67   61.22623.4871
   62.66  623.28   65.64   623.3   71.61  623.65   89.51   623.9   100.7   623.6
  109.09  623.02  113.85  622.89  121.39623.4874  129.22   624.5  135.34   626.5
  141.47  631.09  144.53  632.93  147.59  634.32  150.66  636.24  159.84  639.34
#Mann= 3 , 0 , 0
       0      .1       0   61.22      .1       0  121.39      .1       0
Bank Sta=61.22,121.39
XS Rating Curve= 0 ,0
Exp/Cntr=0.3,0.1

Type RM Length L Ch R = 1 ,2560.316,88.9,91.4,90.97
XS GIS Cut Line= 3
     616407.7906     4341965.608     616353.8284    4342007.8496
     616312.5404    4342044.9832
#Sta/Elev= 30
       0   639.3    2.98  638.91    5.96  637.58    8.94  636.45   11.92  634.88
    14.9  632.78   17.88  630.31   20.86  628.21   23.84  626.27   26.82  624.52
   32.77   621.7   34.39621.1455   35.75  620.68   38.73  620.38   44.69  620.89
   50.65  621.13   59.59   621.3   62.57  621.26   65.55  621.02   68.53  620.99
   69.95621.1456    77.3  622.09   86.07  622.89   88.99  623.02   91.91  623.32
   94.83  624.09   97.76  625.26   103.6     628  118.21  635.15  124.06  639.14
#Mann= 3 , 0 , 0
       0      .1       0   34.39      .1       0   69.95      .1       0
Bank Sta=34.39,69.95
XS Rating Curve= 0 ,0
Exp/Cntr=0.3,0.1

Type RM Length L Ch R = 1 ,2468.92 ,95.43,91.51,94.03
XS GIS Cut Line= 3
        616393.9    4341869.0349     616293.6344      4341943.94
     616249.7018    4341973.5456
#Sta/Elev= 30
       0  639.49    3.05  638.86    6.11  638.53   24.42   635.2   27.47  634.08
   33.58  632.75   48.84  630.86   54.95  629.21      58  627.22   61.05  625.66
   67.16  623.03   70.21  622.03   73.26  621.47   82.42  620.29   87.73619.2277
   91.58  618.79   94.63  618.76   122.1  619.25   128.1  619.19  133.99  618.88
  136.93  619.03  138.01619.2284  145.76  620.55   148.7  621.26  151.64   622.6
  160.47  628.44  163.42  631.19  166.36  633.45  172.25     637  178.13  638.92
#Mann= 3 , 0 , 0
       0      .1       0   87.73      .1       0  138.01      .1       0
Bank Sta=87.73,138.01
XS Rating Curve= 0 ,0
Exp/Cntr=0.3,0.1

Type RM Length L Ch R = 1 ,2377.412,95.29,91.41,88.71
XS GIS Cut Line= 3
     616301.5337    4341795.5423     616229.1695    4341878.3525
     616208.7708    4341898.0166
#Sta/Elev= 30
       0   630.1    3.05  629.72   12.22  629.23   15.27  628.89   24.44  627.31
   27.49   626.5    33.6  625.42   39.71  622.91   42.77  621.48   48.88  617.98
    53.4 616.679   54.99  616.37   58.04  616.13    61.1  616.28   67.21  617.16
   70.26  617.43   82.48  617.57  103.86  616.85  106.92  616.38  109.97  616.12
  112.81  616.37  113.85616.6793  115.64  617.22  118.47  618.86  121.31  619.64
  124.14  620.67  126.97  622.52  132.64  625.79  135.47  627.97  138.31  630.63
#Mann= 3 , 0 , 0
       0      .1       0    53.4      .1       0  113.85      .1       0
Bank Sta=53.4,113.85
XS Rating Curve= 0 ,0
Exp/Cntr=0.3,0.1

Type RM Length L Ch R = 1 ,2286    ,90.33,92.04,91.18
XS GIS Cut Line= 4
     616235.6524    4341708.2297     616184.5484    4341783.1115
     616178.6789    4341800.6348     616148.6035    4341841.9883
#Sta/Elev= 30
       0  630.42    6.04  628.47    9.07  627.67   12.09  626.16   15.11  624.41
   18.13  622.94   21.15  621.66   24.18  620.86    27.2  620.46   30.22  620.38
   33.24  620.14   42.31  618.04   54.39  614.92   57.42  614.71   72.47614.1927
   90.66   613.8  101.22  613.89  109.14  614.11  118.16  613.96  122.77614.1929
  130.19  614.68   133.2  615.08  136.21  616.46  142.22  620.06  145.23  622.38
  148.24  624.49  151.25  626.23  154.26  627.09  157.26  628.19  160.27  629.92
#Mann= 3 , 0 , 0
       0      .1       0   72.47      .1       0  122.77      .1       0
Bank Sta=72.47,122.77
XS Rating Curve= 0 ,0
Exp/Cntr=0.3,0.1

Type RM Length L Ch R = 1 ,2193.958,92.79,90.84,90.43
XS GIS Cut Line= 2
     616140.4022    4341681.2421     616077.6958    4341794.7486
#Sta/Elev= 25
       0  630.28    6.03  628.08   12.06  626.79   18.09  624.04   33.17   618.6
   42.22  614.89   45.24  614.48   51.27  612.66   59.96611.2316   63.33  610.72
   66.35  610.63   78.87611.2314   90.47  611.56   93.49  611.54    96.5  611.89
   99.52  613.46  102.53  616.09  105.55   618.1  111.58  621.61   114.6  623.55
  117.61  625.09  120.63   625.9  123.64  627.55  126.66  629.59  129.68   631.3
#Mann= 3 , 0 , 0
       0      .1       0   59.96      .1       0   78.87      .1       0
Bank Sta=59.96,78.87
XS Rating Curve= 0 ,0
Exp/Cntr=0.3,0.1

Type RM Length L Ch R = 1 ,2103.12 ,33.33,36.06,37.5
XS GIS Cut Line= 3
      616064.202    4341624.8858     616020.0474    4341711.1727
     616008.6194    4341752.6743
#Sta/Elev= 30
       0  630.21    6.06  628.81   15.15  626.44   18.17  626.26   24.23  625.26
   27.26  624.96   30.29  624.98   39.38   625.8   45.44  625.89   54.52  624.42
   60.58  622.52   63.61  621.33    72.7  616.98   78.75  613.07   81.78  610.76
   84.54609.1022   84.81  608.94   87.84  608.47   90.87  608.14    93.9  608.12
  108.41   608.6  111.31609.1028  114.15  611.26  117.02  614.21  119.89   616.3
  122.76  616.84  125.63  618.42  131.37  623.02  134.23  625.16  139.97   629.1
#Mann= 3 , 0 , 0
       0      .1       0   84.54      .1       0  111.31      .1       0
Bank Sta=84.54,111.31
XS Rating Curve= 0 ,0
Exp/Cntr=0.3,0.1

Type RM Length L Ch R = 1 ,2067.061,31.92,36.62,37.95
XS GIS Cut Line= 5
     616044.5647    4341616.7382     616022.4058    4341658.7409
     615997.9318    4341687.1836     615980.1551    4341712.1041
     615968.9103    4341733.5354
#Sta/Elev= 30
       0  630.11   11.87  624.77   14.84  623.88   17.81   623.2   20.78  622.85
   23.74  622.67   32.65  622.42   41.55  622.33   47.49  622.09   50.38  621.79
   53.26  621.19   56.15  619.72   59.03  617.88   64.81  615.28   67.69  614.34
   76.35  608.96   76.89608.8255   79.24  608.24   85.01  608.59   88.07  608.61
   97.26  608.56  103.38  608.34  108.71608.8264  112.56  609.04  115.62   610.1
  118.65   612.7   124.7  619.16  127.72  621.99  133.78  626.61  139.83  631.02
#Mann= 3 , 0 , 0
       0      .1       0   76.89      .1       0  108.71      .1       0
Bank Sta=76.89,108.71
XS Rating Curve= 0 ,0
Exp/Cntr=0.3,0.1

Type RM Length L Ch R = 1 ,2030.443,25.42,18.76,17.25
XS GIS Cut Line= 6
     616021.4302    4341607.5935     616002.5124     4341639.079
      615976.054    4341669.1093     615963.8832    4341679.0311
     615948.9342    4341688.6885     615934.6466    4341716.7343
#Sta/Elev= 30
       0  629.07    6.12  626.67   12.24  625.31    15.3  624.06   21.43  621.23
   24.49  620.83   33.67  620.01   39.59  619.13   42.45  617.82   45.31  616.05
   48.17  615.17   62.46  609.02   65.32  608.08   68.18  607.99    73.9   608.6
   84.61  608.38   87.22  608.18   92.06606.9738   95.42  606.49   98.39  606.41
   104.8 606.973  107.29  607.51  110.25  609.11  113.12  611.44  124.56   621.8
  127.42  624.17  130.28     626  136.01  629.27  138.87  629.85  141.73  630.73
#Mann= 3 , 0 , 0
       0      .1       0   92.06      .1       0   104.8      .1       0
Bank Sta=92.06,104.8
XS Rating Curve= 0 ,0
Exp/Cntr=0.3,0.1

Type RM Length L Ch R = 1 ,2011.68 ,86.01,91.43,93.06
XS GIS Cut Line= 3
     616000.7019    4341597.1045     615955.4715    4341650.1881
     615919.8794    4341705.8001
#Sta/Elev= 30
       0  629.44    3.03  628.46    6.06  627.69   15.16  625.62   18.19  624.63
   21.23  623.44   27.29  620.57   30.32  620.23   39.42  613.73   45.48  609.12
   48.51   607.7   51.55  607.09   54.58  606.87   66.71  607.55   81.74  607.86
   84.75  607.23   85.99606.8084   87.75  606.21   90.75  605.79   93.75  606.07
   97.11606.8069   99.75  607.45  102.75  608.81  105.75  611.07  108.76  612.91
  111.76  615.62  114.76  617.15  120.76  621.22  123.76  622.89  135.77  628.96
#Mann= 3 , 0 , 0
       0      .1       0   85.99      .1       0   97.11      .1       0
Bank Sta=85.99,97.11
XS Rating Curve= 0 ,0
Exp/Cntr=0.3,0.1

Type RM Length L Ch R = 1 ,1920.249,93.78,91.45,89.78
XS GIS Cut Line= 3
     615989.6423    4341519.9518     615872.6015    4341615.2785
     615843.8515    4341642.1699
#Sta/Elev= 30
       0  619.36    6.04  619.98   12.08  620.33   18.11  618.32   21.13  618.22
   24.15  617.69   27.17  616.88   42.27  617.41    48.3  617.24   51.32  616.56
   54.34  614.63    63.4  611.96   75.47  607.49   78.49  606.83   88.78  605.15
   90.57  604.99  114.72  604.83  123.78  605.29  138.87   605.7  147.93  605.39
  153.98  604.57  157.01  604.58  160.03  605.15  163.06  606.04  166.09  607.79
  169.12  610.84  172.15  613.18  181.23  617.34  184.26  617.87  190.32  620.53
#Mann= 3 , 0 , 0
       0      .1       0   88.78      .1       0  160.03      .1       0
Bank Sta=88.78,160.03
XS Rating Curve= 0 ,0
Exp/Cntr=0.3,0.1

Type RM Length L Ch R = 1 ,1828.8  ,95.48,91.44,88.85
XS GIS Cut Line= 3
     615875.8838    4341486.4373     615824.1715    4341540.3501
     615787.3799    4341574.8744
#Sta/Elev= 28
       0  611.92    2.99  608.97    5.98  606.69    8.96  604.73   11.95  603.39
   14.94  602.78   16.04602.6476   20.92  602.12   23.91  602.11   29.88  602.47
   38.85  602.83   47.81  602.96   53.79  602.92   56.78   602.8   59.76  602.64
   65.74  602.14   68.73  602.31   71.81602.6472    74.7  602.88   83.61   603.3
   95.48  603.59   98.45  603.88  101.42  604.52  104.38  605.26  110.32  606.32
  113.29  607.16  116.25  608.21  125.16  611.83
#Mann= 3 , 0 , 0
       0      .1       0   16.04      .1       0   71.81      .1       0
Bank Sta=16.04,71.81
XS Rating Curve= 0 ,0
Exp/Cntr=0.3,0.1

Type RM Length L Ch R = 1 ,1737.36 ,92.75,91.44,88.33
XS GIS Cut Line= 4
     615792.6457    4341420.4994     615771.0469    4341453.5546
     615763.5456    4341470.0554     615721.1458    4341535.4724
#Sta/Elev= 29
       0  612.96    6.07  607.26    9.11  604.62   12.15  602.18   15.19   600.3
   18.22  600.04   20.89598.4503   21.26  598.23    24.3   597.7   27.34  597.95
   30.78  598.45   45.53  600.01   48.55  600.11   57.61  600.02   60.61   600.1
   69.61  600.52    87.6  601.16   93.59  601.25   99.59  601.46  102.59  601.66
  105.58  602.23  108.58  603.21  111.58  604.37  117.58  606.45  120.58   607.7
  126.57  609.84  129.57  611.13  132.57  611.65  135.57  612.54
#Mann= 3 , 0 , 0
       0      .1       0   20.89      .1       0   30.78      .1       0
Bank Sta=20.89,30.78
XS Rating Curve= 0 ,0
Exp/Cntr=0.3,0.1

Type RM Length L Ch R = 1 ,1645.92 ,54.04,54.65,48.73
XS GIS Cut Line= 5
     615688.9707    4341398.2952     615678.0866    4341435.8353
      615672.131    4341446.8198     615672.8311    4341459.0833
     615640.3894    4341517.6742
#Sta/Elev= 30
       0  612.55    3.01  608.89    6.01  604.77    9.02  600.34   11.93 597.227
   15.03  596.07   24.05  596.87   26.13597.2224   27.06  597.38   30.07  597.39
   33.07  597.58   36.08  598.19   39.09   598.5   57.72  598.71   69.95  599.14
   76.04  599.48   79.09   599.8   82.13  600.78   85.17  601.98   88.22   602.7
   91.26  603.14   94.31  603.52   100.4  602.88  106.48  603.49  109.53  604.21
  112.57  605.35   121.7  609.85  124.75  611.08  127.79  611.41  130.84  612.33
#Mann= 3 , 0 , 0
       0      .1       0   11.93      .1       0   26.13      .1       0
Bank Sta=11.93,26.13
XS Rating Curve= 0 ,0
Exp/Cntr=0.3,0.1

Type RM Length L Ch R = 1 ,1591.275,35.03,36.82,41.31
XS GIS Cut Line= 4
     615628.0884    4341377.7909     615623.5007    4341450.0155
     615624.4929    4341462.5833     615613.6706    4341506.9548
#Sta/Elev= 30
       0  613.31    6.03  609.07    9.05  607.49   15.08     606   18.09  605.96
   27.14  603.95   30.15  602.98   33.17  601.27   38.85596.6667    39.2  596.39
   42.22  595.78   54.28  596.39   66.84596.6683   72.37  596.92   77.41  597.36
   79.93  597.41   82.46  597.81   88.02  598.23   91.07  598.33   97.16  598.29
   100.2  598.51  103.25  599.62  106.29  601.43  109.34  602.52  112.38  603.18
  115.43  604.35  118.47  605.33  121.51  606.56  124.56  608.02  130.65   611.6
#Mann= 3 , 0 , 0
       0      .1       0   38.85      .1       0   66.84      .1       0
Bank Sta=38.85,66.84
XS Rating Curve= 0 ,0
Exp/Cntr=0.3,0.1

Type RM Length L Ch R = 1 ,1554.456,61.83,62.47,64.13
XS GIS Cut Line= 4
     615605.2416    4341367.6573      615585.766    4341446.5857
     615563.8777    4341501.4719     615553.1186    4341538.0493
#Sta/Elev= 30
       0  614.09    3.01  612.85    9.03  609.92   12.04  608.79   18.07   607.2
    27.1  605.39   39.14  604.01   42.15  603.57   45.16  602.75   48.18  600.52
   51.19  597.48   53.88596.0233    54.2  595.85   57.21  595.56   66.24  595.47
   78.28  595.54   82.11596.0229   90.16  597.85   93.11  598.84   96.07  600.44
   99.02  600.62  104.93  603.67  107.89  604.52  110.84  605.06  128.57  607.77
  134.48  608.19  143.32  609.46  160.92   611.2  166.78  611.36  178.51  612.67
#Mann= 3 , 0 , 0
       0      .1       0   53.88      .1       0   82.11      .1       0
Bank Sta=53.88,82.11
XS Rating Curve= 0 ,0
Exp/Cntr=0.3,0.1

Type RM Length L Ch R = 1 ,1491.988,28.15,28.93,31.79
XS GIS Cut Line= 5
     615544.1256    4341372.6248     615533.8399    4341402.0531
     615530.1886    4341415.8644     615529.0245    4341423.5902
      615507.064    4341467.5111
#Sta/Elev= 21
       0  602.79    2.83  602.38    5.67   602.1   22.67  598.82   25.51  598.21
   28.34  597.29   31.17     596   33.88595.1567   48.06   594.4   50.67   594.4
    58.2595.1578   65.55  595.87   74.76  596.11   77.83  596.38   80.89  596.54
   87.03  597.26    90.1  598.08   93.17  599.28   96.24  600.85   99.31  602.94
  102.38  605.66
#Mann= 3 , 0 , 0
       0      .1       0   33.88      .1       0    58.2      .1       0
Bank Sta=33.88,58.2
XS Rating Curve= 0 ,0
Exp/Cntr=0.3,0.1

Type RM Length L Ch R = 1 ,1463.059,91.19,91.47,91.46
XS GIS Cut Line= 3
     615529.8903    4341353.8218      615501.548    4341408.1225
     615485.2282    4341435.8734
#Sta/Elev= 22
       0  603.36    3.06  602.42    9.19  600.74   15.31  599.28   18.38  598.64
    24.5  597.54   27.56  597.16   30.63  596.92   46.63594.2505      49  593.84
   52.06  593.45   55.13  593.47   58.19   593.9   59.86594.2493   64.18  595.03
   67.11  595.18   70.03   595.5   78.81  596.73   81.74  597.26   84.67  598.24
   87.59  599.55   93.45  602.36
#Mann= 3 , 0 , 0
       0      .1       0   46.63      .1       0   59.86      .1       0
Bank Sta=46.63,59.86
XS Rating Curve= 0 ,0
Exp/Cntr=0.3,0.1

Type RM Length L Ch R = 1 ,1371.584,91.92,91.42,89.33
XS GIS Cut Line= 4
     615447.2079    4341322.0717     615421.5115    4341362.9356
     615411.1193    4341385.2128     615405.3335    4341422.4795
#Sta/Elev= 28
       0  603.12    3.02   602.1    6.03  600.98   12.07  599.73   21.12  596.25
   27.15   593.8   30.17  592.83   33.68 591.897    36.2  591.47   38.87  591.45
   42.24  591.52   48.27  591.48   51.34  591.58   57.49  591.48   61.41591.8962
   63.64  592.07   66.71  592.19   78.66  592.47   84.46  592.53   87.36  593.06
   90.26  594.73   93.16  596.64   96.06   597.7   98.96  598.48  101.86  599.45
  104.76  600.69  107.67  602.18  110.57  603.99
#Mann= 3 , 0 , 0
       0      .1       0   33.68      .1       0   61.41      .1       0
Bank Sta=33.68,61.41
XS Rating Curve= 0 ,0
Exp/Cntr=0.3,0.1

Type RM Length L Ch R = 1 ,1280.16 ,12.82,12.17,12.25
XS GIS Cut Line= 4
     615356.5879    4341292.9675     615339.1373    4341330.5705
     615334.7182    4341346.1461      615308.788    4341410.0052
#Sta/Elev= 28
       0   605.8    2.96  602.67    5.92  599.64    8.88  597.18   11.84     595
   14.81   593.1   17.77  591.53   20.73  591.05   23.69  590.35   26.27589.8358
   29.61  589.59   38.49  589.65   44.15  589.34   60.64  589.21   63.64  589.26
   70.45589.8365   72.63  589.96   81.62  590.07    96.6  590.09    99.6  590.33
  102.59  590.83  105.59  591.68  108.59  592.97  111.58  594.74  114.58  597.15
  120.57  602.44  123.57     603  126.57  604.62
#Mann= 3 , 0 , 0
       0      .1       0   26.27      .1       0   70.45      .1       0
Bank Sta=26.27,70.45
XS Rating Curve= 0 ,0
Exp/Cntr=0.3,0.1

Type RM Length L Ch R = 1 ,1267.992,11.78,11.5,12.51
XS GIS Cut Line= 5
     615345.5948    4341286.4769     615327.8147     4341324.577
     615324.3222    4341340.2932     615305.4309    4341380.6158
     615279.0784    4341398.7134
#Sta/Elev= 27
       0  606.58    6.01  601.71   12.01  597.04   15.02  594.88   18.02  592.88
   21.02  591.11   24.03  590.06   27.03  589.81   33.04   589.9   37.84 589.796
   42.04  589.57   44.73  589.32   47.41  589.23   52.78   589.3   70.02  589.21
   78.92  589.35   89.24 589.796   96.74  590.21    99.7  590.78  102.67  591.65
  105.58  593.15  108.49  594.87   114.3  598.52  125.92  605.24  128.83  607.93
  131.73   609.7  134.64   611.2
#Mann= 3 , 0 , 0
       0      .1       0   37.84      .1       0   89.24      .1       0
Bank Sta=37.84,89.24
XS Rating Curve= 0 ,0
Exp/Cntr=0.3,0.1

Type RM Length L Ch R = 1 ,1256.492,61.35,67.77,71.18
XS GIS Cut Line= 6
     615338.2923    4341279.6506     615319.0835    4341313.7819
     615313.8976    4341334.2078     615307.4418    4341346.1141
     615295.4896    4341365.6369     615268.2904    4341384.5811
#Sta/Elev= 30
       0  607.17    3.01  604.73    6.03  603.93    9.04  601.82   21.09  593.02
    24.1  591.06   27.11  590.12   30.13  589.95   44.29589.5731   47.45  589.37
   50.01  589.03   52.57  588.93   57.69  589.44   60.25  589.62   65.67  589.57
    73.8  589.27   85.24  589.21   90.96  589.35    92.9589.5731   93.83  589.68
   96.69  590.23    99.7  591.25  102.71  592.76  105.73  595.13  108.74  597.91
  117.78  604.08  120.79  606.46  123.81  608.18  126.82  609.31  129.83  611.22
#Mann= 3 , 0 , 0
       0      .1       0   44.29      .1       0    92.9      .1       0
Bank Sta=44.29,92.9
XS Rating Curve= 0 ,0
Exp/Cntr=0.3,0.1

Type RM Length L Ch R = 1 ,1188.72 ,16.7,16.84,16.91
XS GIS Cut Line= 2
     615297.4999    4341256.7018      615225.898    4341328.3039
#Sta/Elev= 18
       0  602.49    6.14  600.09   18.41   591.4   21.48  589.43   24.55  588.17
   27.62  587.65   42.96  587.13   55.41586.3271   64.44  585.75   67.51  585.85
   71.03586.3276   76.71  587.09   79.78  587.94   82.85  589.74   88.99  594.02
   95.12  599.84   98.19  601.45  101.26  602.62
#Mann= 3 , 0 , 0
       0      .1       0   55.41      .1       0   71.03      .1       0
Bank Sta=55.41,71.03
XS Rating Curve= 0 ,0
Exp/Cntr=0.3,0.1

Type RM Length L Ch R = 1 ,1171.883,16.29,16.72,16.96
XS GIS Cut Line= 2
     615282.5145    4341248.7437     615214.3576    4341315.4188
#Sta/Elev= 21
       0  601.75    2.98  598.85    5.96  596.66    14.9  590.48   17.88  588.98
   20.86  588.31   23.84  587.32   26.82   586.8   35.95585.8119   38.73  585.56
   41.71  585.48   56.61  585.44   59.59  585.45   64.23585.8127   65.55  585.95
   68.53  586.07   71.51   586.4   74.49   587.5   77.47  589.43   92.37  599.74
   95.35  602.42
#Mann= 3 , 0 , 0
       0      .1       0   35.95      .1       0   64.23      .1       0
Bank Sta=35.95,64.23
XS Rating Curve= 0 ,0
Exp/Cntr=0.3,0.1

Type RM Length L Ch R = 1 ,1155.16 ,15.43,15.76,15.93
XS GIS Cut Line= 2
     615270.2378    4341240.0654     615202.2926    4341301.8721
#Sta/Elev= 21
       0  600.86    9.19  594.57   12.25  592.35   15.31  589.63   18.37  587.82
   21.43  586.66   24.49  586.17   27.28585.8701   33.68  585.39   42.86  585.18
   55.31  585.19   58.17  585.26    64.3   585.6   67.44585.8691   70.42  586.95
   73.48  589.79   76.54  592.08   82.67   596.5   85.73  598.48   88.79  599.49
   91.85  601.66
#Mann= 3 , 0 , 0
       0      .1       0   27.28      .1       0   67.44      .1       0
Bank Sta=27.28,67.44
XS Rating Curve= 0 ,0
Exp/Cntr=0.3,0.1

Type RM Length L Ch R = 1 ,1139.404,16.76,19.67,21.22
XS GIS Cut Line= 4
     615268.9678    4341236.0437     615233.4077     4341252.977
     615210.7593    4341272.4504     615189.8043    4341291.9238
#Sta/Elev= 24
       0  601.54    3.03  600.32    6.06  598.73    9.09  596.62   12.12  594.68
   15.15  592.39   18.18  589.83   21.21  587.72   24.24  586.74   27.27  586.29
    30.3  585.98   34.11585.7491   45.36  585.32   57.31  584.99   63.28  585.19
   66.27   585.4   69.69585.7491   72.12  586.14   74.98  587.15   77.84  588.93
   83.56  592.77   89.28  597.25   92.14   600.2   97.86  604.42
#Mann= 3 , 0 , 0
       0      .1       0   34.11      .1       0   69.69      .1       0
Bank Sta=34.11,69.69
XS Rating Curve= 0 ,0
Exp/Cntr=0.3,0.1

Type RM Length L Ch R = 1 ,1119.734,24.5,22.46,22.14
XS GIS Cut Line= 4
     615291.8278    4341216.9936     615225.9993    4341239.8537
     615198.6943    4341253.4004     615174.1409    4341267.3704
#Sta/Elev= 30
       0  603.57    6.06  602.86    9.09  602.04   15.15  601.33   21.21  600.51
   24.24  600.32   27.27  599.95    30.3  598.76   36.36  595.84   39.39  594.02
   42.42  592.32   45.45  590.37   48.48  588.22   51.51  586.98   54.54  586.48
   57.57   586.2   75.79585.4094   84.93  584.98   91.02   584.6   94.07  584.54
   97.12  585.13   98.02585.4103  100.17  586.08  102.99  587.19  105.82  588.68
  117.12  595.32  119.94  597.15  122.77  600.07  125.59  601.93  128.42  603.64
#Mann= 3 , 0 , 0
       0      .1       0   75.79      .1       0   98.02      .1       0
Bank Sta=75.79,98.02
XS Rating Curve= 0 ,0
Exp/Cntr=0.3,0.1

Type RM Length L Ch R = 1 ,1097.277,38.37,38.19,38.11
XS GIS Cut Line= 2
     615238.8481    4341203.6705     615163.4417    4341249.9726
#Sta/Elev= 25
       0  602.44    3.05  600.41     6.1  599.56    9.15  598.45   12.21  596.19
   15.26  593.55   21.36  589.52   24.41  587.85   27.46  586.38   30.51   585.5
   32.59585.1522   36.62  584.57   39.67  584.29   45.77  584.22   51.87  584.22
   54.92  584.37   57.98585.1545   61.03  586.53   64.08  588.41   67.13  591.12
   70.18  592.92   73.23  594.87   79.33  597.55   85.44  601.06   88.49  602.66
#Mann= 3 , 0 , 0
       0      .1       0   32.59      .1       0   57.98      .1       0
Bank Sta=32.59,57.98
XS Rating Curve= 0 ,0
Exp/Cntr=0.3,0.1

Type RM Length L Ch R = 1 ,1059.083,48.38,53.24,54.83
XS GIS Cut Line= 3
     615220.3227    4341176.1243     615187.7789    4341189.8826
     615143.5934    4341218.4577
#Sta/Elev= 25
       0  603.39    2.94  601.42   11.78  596.32   14.72   592.6   17.67  590.38
   20.61  588.44   23.56  586.62    26.5   585.2   28.22584.8197   29.44  584.55
   32.39  584.43   35.33  584.42    44.1   584.6   47.03  584.56   49.95  584.36
   52.87  583.95    55.8  584.12   57.41584.8203   58.72  585.39   61.64  587.79
   64.57  590.92   70.41  594.36   79.18  599.66   85.03  602.55   87.95  603.87
#Mann= 3 , 0 , 0
       0      .1       0   28.22      .1       0   57.41      .1       0
Bank Sta=28.22,57.41
XS Rating Curve= 0 ,0
Exp/Cntr=0.3,0.1

Type RM Length L Ch R = 1 ,1005.84 ,92.73,91.44,89.95
XS GIS Cut Line= 4
     615195.7337      4341143.57     615163.1251    4341148.6348
     615154.1927     4341148.861      615108.739    4341159.1432
#Sta/Elev= 23
       0  593.96       3   591.1       6  588.05       9  586.22      12  584.62
      15  583.61      18  583.19      24  582.76      27  582.41      33  582.06
    38.2581.6171   41.93  581.23   44.85  581.12   47.76  581.23   50.32581.6171
    56.5  582.79   62.32  584.08   65.24  585.17   68.15  586.55   73.97  588.18
   76.89  589.22   85.62  592.97   88.54  595.12
#Mann= 3 , 0 , 0
       0      .1       0    38.2      .1       0   50.32      .1       0
Bank Sta=38.2,50.32
XS Rating Curve= 0 ,0
Exp/Cntr=0.3,0.1

Type RM Length L Ch R = 1 ,914.4   ,90.46,91.44,93.19
XS GIS Cut Line= 4
     615177.4587    4341048.8242     615131.5531    4341061.9401
     615114.7488    4341068.7747     615043.1222     4341076.593
#Sta/Elev= 25
       0  593.75    2.98  591.51    5.97  589.43    8.95  587.55   14.92  583.97
    17.9  581.81   20.89  581.46   29.84  580.68    33.4580.2872   35.81  579.86
   38.79  579.56   41.77  579.52   57.89580.2877   77.89  581.28    83.9  581.65
   98.91  581.93  104.91  582.19  107.91  582.73  113.92  584.28  116.92  584.84
  119.92   585.6  125.93  588.28  128.93  589.74  134.93  592.05  137.94  593.37
#Mann= 3 , 0 , 0
       0      .1       0    33.4      .1       0   57.89      .1       0
Bank Sta=33.4,57.89
XS Rating Curve= 0 ,0
Exp/Cntr=0.3,0.1

Type RM Length L Ch R = 1 ,822.9601,94.7,91.44,91.53
XS GIS Cut Line= 3
     615173.2853     4340970.841     615129.1365    4340970.3694
     615070.6689    4340976.7476
#Sta/Elev= 22
       0  594.76    2.94   592.2    5.89  590.13   17.66  583.26    20.6  581.19
   23.55  579.62   26.49  579.32   35.32  578.95   38.26  578.71   41.21   578.3
   44.15  577.52   46.03577.2834   50.03  576.95   52.97  576.94   70.62  577.08
   73.66577.2849    76.5  577.99   79.44  579.48   82.38  582.12   85.32   584.6
  100.03  591.79  102.97  593.46
#Mann= 3 , 0 , 0
       0      .1       0   46.03      .1       0   73.66      .1       0
Bank Sta=46.03,73.66
XS Rating Curve= 0 ,0
Exp/Cntr=0.3,0.1

Type RM Length L Ch R = 1 ,731.52  ,89.13,91.44,92.71
XS GIS Cut Line= 3
     615166.9774    4340877.7464     615103.4429    4340881.0556
     615068.7178    4340886.3772
#Sta/Elev= 20
       0  587.24    3.03     586    6.06  583.76    9.09  582.28   21.21  577.62
   24.24  576.53   27.27  575.86    30.3  575.62   33.54575.5337   48.47  575.01
   54.53  574.91   60.59  575.07   66.94 575.534   69.48  575.69   75.33  575.67
   78.26  575.95   81.19  576.64   84.11  577.64   87.04  579.69   98.75  584.16
#Mann= 3 , 0 , 0
       0      .1       0   33.54      .1       0   66.94      .1       0
Bank Sta=33.54,66.94
XS Rating Curve= 0 ,0
Exp/Cntr=0.3,0.1

Type RM Length L Ch R = 1 ,640.08  ,92.13,91.44,86.51
XS GIS Cut Line= 4
     615167.0769    4340794.9635     615126.6832    4340791.4864
     615112.2898    4340789.2606     615034.5203    4340787.2906
#Sta/Elev= 26
       0  583.81     2.9   583.1    5.79  582.14    8.69  581.02   11.58  579.79
   14.48     578   17.38  576.04   20.27  574.86   23.17  573.98   24.69573.7117
   26.06  573.47   28.96  573.31   31.86  573.29   52.19  573.37   65.63573.7113
   73.06  573.92   79.04  574.25      94  574.81   99.99  574.81  105.97  574.44
  108.97  574.71  111.96  575.73  114.95  577.29  117.94  579.84  123.93  582.46
   132.9  586.67
#Mann= 3 , 0 , 0
       0      .1       0   24.69      .1       0   65.63      .1       0
Bank Sta=24.69,65.63
XS Rating Curve= 0 ,0
Exp/Cntr=0.3,0.1

Type RM Length L Ch R = 1 ,548.64  ,88.77,91.44,93.32
XS GIS Cut Line= 4
     615195.8371    4340697.0807     615113.1244    4340700.2574
     615058.4091    4340708.6752     615021.7694    4340710.8988
#Sta/Elev= 26
       0  583.95    6.13  580.69     9.2  579.23   18.39  575.44   21.46  574.71
   27.59   573.5   30.66  573.03   36.79  572.31   55.16571.2011   61.31  570.95
   73.58  570.81   82.77  570.86   94.73571.2012  111.91  572.07  117.74   572.5
  135.22  573.48  138.13  573.74  150.37  574.27  153.43  574.32  156.49  574.27
  159.55  575.32   162.6  579.68  165.66  582.22  168.72  583.25  171.78  583.91
  174.84  585.01
#Mann= 3 , 0 , 0
       0      .1       0   55.16      .1       0   94.73      .1       0
Bank Sta=55.16,94.73
XS Rating Curve= 0 ,0
Exp/Cntr=0.3,0.1

Type RM Length L Ch R = 1 ,457.2   ,45.57,91.44,92.07
XS GIS Cut Line= 5
     615217.7698    4340675.7966     615143.9787    4340611.6466
     615102.7611    4340610.9018     615074.5517    4340612.8252
      615004.803    4340614.5877
#Sta/Elev= 30
       0  584.54    3.06  583.05    6.11  582.15    9.17  581.61   15.28   578.6
   18.33  576.74   21.39  575.68   39.72  572.61   42.78  571.89   45.83   571.5
   67.22  570.31   85.55  569.44   88.61  569.44   97.78  568.84  142.47566.7296
  161.62  566.41  173.34  566.48  178.54566.7297  188.51  567.89  191.54  568.61
  194.58  569.07  206.71  570.33  209.75  570.35  212.78  571.84  215.81   573.7
  218.85  575.24  227.95  579.44  230.98  581.88  234.01  584.04  237.05   585.6
#Mann= 3 , 0 , 0
       0      .1       0  142.47      .1       0  178.54      .1       0
Bank Sta=142.47,178.54
XS Rating Curve= 0 ,0
Exp/Cntr=0.3,0.1
