HEC-RAS study MinearRun.prj: MinearRun

--- MinearRun.g01 (geometry) --- (continued)

Type RM Length L Ch R = 1 ,365.76  ,45.19,91.49,77.95
XS GIS Cut Line= 6
     615230.7431    4340673.5738      615131.874    4340566.1382
     615115.2052    4340565.3444      615093.785    4340520.9884
     615068.3662    4340520.5849     614981.0612    4340529.6256
#Sta/Elev= 30
       0  586.34    3.04  584.83    6.08  583.68    9.13   582.9   21.29  576.76
   24.33  575.71    36.5   573.1   42.58   572.2   48.67  571.96   76.04  569.46
    94.3  568.06  106.46  567.81  127.75  567.96  151.57  567.25  172.37565.4352
  185.87  564.45  194.57  564.36  197.46   564.4  203.26  565.14  206.16  565.26
  231.41565.4356  261.59  565.66  282.77  566.65   285.8   566.9  288.82  567.54
  294.88  570.06  303.96  574.56  310.01  579.31  322.12  584.76  325.14  586.82
#Mann= 3 , 0 , 0
       0      .1       0  172.37      .1       0  231.41      .1       0
Bank Sta=172.37,231.41
XS Rating Curve= 0 ,0
Exp/Cntr=0.3,0.1

River Reach=Mill Run(Minear),1
Reach XY= 30
     615073.5775    4340448.2522     615069.0555    4340444.5961
     615064.5335    4340440.9401     615057.7506    4340435.4559
     615048.7066    4340428.1438     615034.0342    4340424.9478
     615031.0998    4340424.3087     615025.2308    4340423.0303
     614998.8206    4340417.2775     614995.8861    4340416.6384
     614978.2793    4340412.8032      614934.559    4340401.0659
     614925.6513    4340400.2721     614922.6821    4340400.0076
     614904.8668      4340398.42     614901.8976    4340398.1555
     614887.0514    4340396.8325     614884.0822     4340396.568
     614866.2669    4340394.9804     614863.2977    4340394.7159
       614854.39    4340393.9221     614845.5645    4340393.8978
     614842.6227    4340393.8898     614827.9136    4340393.8493
     614824.9718    4340393.8413     614807.3209    4340393.7927
     614804.3791    4340393.7847     614795.5536    4340393.7604
     614793.7014    4340393.3115     614791.8493    4340392.8625

Type RM Length L Ch R = 1 ,274.2707,93.1,91.6,76.07
XS GIS Cut Line= 5
     615087.3297    4340401.9924     615052.4042    4340445.5803
     615043.7345    4340443.1728      615038.972     4340452.301
     614986.0891    4340499.7599
#Sta/Elev= 24
       0  576.55    5.88   574.8    8.82  573.81   20.58  569.39   23.52  568.87
   32.34  565.93   35.28  565.04   36.47564.7769   38.22  564.39   41.16  564.11
   49.97  564.21   64.85  564.57   75.15  564.96   89.95  565.38  101.79  564.91
  104.75  564.75  110.68  564.27   113.9564.7762  119.56  565.94  122.52  566.38
  128.44  567.43   131.4  568.43  134.36  569.96   146.2  576.49
#Mann= 3 , 0 , 0
       0      .1       0   36.47      .1       0   113.9      .1       0
Bank Sta=36.47,113.9
XS Rating Curve= 0 ,0
Exp/Cntr=0.3,0.1

Type RM Length L Ch R = 1 ,182.6682,91.79,91.23,89.94
XS GIS Cut Line= 3
     614985.7295    4340360.7173     614967.9515    4340429.9711
       614953.22    4340460.3458
#Sta/Elev= 22
       0  576.82    5.96   574.2    8.94  573.07   11.92  572.81   17.87  570.14
   20.85  568.54   23.83  566.39   26.81  564.07    29.7 562.499   32.77  561.94
   53.62  561.82   62.56  561.94    71.5  562.35   74.57  562.37   77.21 562.499
   80.71  562.65   83.78  563.13   86.84  564.23   89.91  565.62   92.98  567.24
   96.05  569.17  105.26  575.37
#Mann= 3 , 0 , 0
       0      .1       0    29.7      .1       0   77.21      .1       0
Bank Sta=29.7,77.21
XS Rating Curve= 0 ,0
Exp/Cntr=0.3,0.1

Type RM Length L Ch R = 1 ,91.44003,35.79,60.98,60.98
XS GIS Cut Line= 4
     614930.6961    4340336.3756     614890.5713    4340365.3014
     614883.8379    4340387.8394     614879.1706    4340440.2164
#Sta/Elev= 26
       0  575.46    2.91  574.53    5.82   573.3   11.64  570.57   17.46  567.31
   20.37  566.39   23.28  565.74   26.19  564.52    29.1  563.02   32.15562.0641
   34.92  561.75   61.23  561.49   70.05  561.46   78.83  561.54   84.67  561.37
   87.59  561.58   90.21562.0645   93.44  562.74   96.36  563.21   99.28  563.34
   102.2  563.59  105.12  564.04  108.04  564.95  110.96  566.63  119.73  573.25
  125.57  577.36
#Mann= 3 , 0 , 0
       0      .1       0   32.15      .1       0   90.21      .1       0
Bank Sta=32.15,90.21
XS Rating Curve= 0 ,0
Exp/Cntr=0.3,0.1

Type RM Length L Ch R = 1 ,30.45887,6990.96,39.6,39.9
XS GIS Cut Line= 6
     614925.4365    4340334.9901     614822.4798    4340388.6715
     614824.8946    4340432.5554     614852.3452    4340490.1024
     614860.9442    4340522.1832     614852.3452    4340567.8239
#Sta/Elev= 30
       0  575.53     2.9  574.22     5.8  572.32   20.29  566.02   28.44562.0888
   31.88  561.67   49.27  561.59   58.15  560.59      70  560.47  116.22  561.28
  160.47   560.9  166.36  561.35  169.46562.0922  175.19  564.25  184.03   566.1
  195.64  569.53  204.22  572.63  207.07  574.37  215.65  576.78  224.23  579.74
  236.31  583.11  242.35  584.04  257.45  589.54   263.2  590.82  268.96  592.58
  274.71  593.41  286.32  597.85  292.27  599.13  301.19  602.82  304.16  602.93
#Mann= 3 , 0 , 0
       0      .1       0   28.44      .1       0  169.46      .1       0
Bank Sta=28.44,169.46
XS Rating Curve= 0 ,0
Exp/Cntr=0.3,0.1

Type RM Length L Ch R = 1 ,19.92903,6980.35,19.93,21.72
XS GIS Cut Line= 6
     614922.5719    4340334.5377     614835.8678    4340372.1615
     614819.6753     4340380.099     614811.7025     4340388.149
     614816.2665    4340433.4788      614814.044    4340466.4989
#Sta/Elev= 30
       0  574.85    3.05  573.04     6.1  571.63   18.29  566.53   21.34   565.1
   24.39  562.84   26.44562.0334   27.44  561.64   45.73  561.58   48.78  560.95
   51.83  560.61   64.03  561.23   94.52  561.27  100.53  561.05  109.54  561.56
  118.21  561.64  123.88  561.96  135.75  561.97  146.87  560.98  149.65   560.9
  163.86  560.93  169.55  561.23  173.86562.0355  175.57  562.49  181.58  564.92
  184.59  565.85  190.61  566.77  193.62  567.73  196.63  569.02  202.64  572.34
#Mann= 3 , 0 , 0
       0      .1       0   26.44      .1       0  173.86      .1       0
Bank Sta=26.44,173.86
XS Rating Curve= 0 ,0
Exp/Cntr=0.3,0.1

River Reach=Stump Run       ,1
Reach XY= 30
     613750.0511    4341774.4173     613773.0699    4341716.8703
     613820.1658    4341679.8815 613863.137906794341604.96250459
613908.6759792654341555.33853266613904.393046605 4341540.2789233
613914.3083790824341522.16844422     613968.7296    4341486.6824
     614025.4829    4341393.0197     614033.4204    4341326.7414
      614052.735    4341281.6299     614049.8412    4341266.6644
     614034.5615    4341251.6823      614044.533    4341195.2962
     614076.6799     4341168.388     614110.6789    4341153.6375
     614177.9415    4341073.7948     614274.7209    4340915.1812
     614364.4148    4340844.9342     614479.9057    4340778.2591
     614486.6526    4340756.4309     614502.0391    4340741.6855
 614513.684223124340701.91768147     614577.8297    4340612.2957
     614661.2779    4340536.1649     614681.1217    4340500.8429
     614737.0812    4340434.9615     614753.2637    4340398.2811
        614772.8    4340388.1302     614791.8493    4340392.8625

Type RM Length L Ch R = 1 ,1828.007,86.32,91.67,99.41
XS GIS Cut Line= 3
     613808.2343    4341774.1507     613738.8208    4341746.7557
     613700.6979    4341719.9217
#Sta/Elev= 26
       0  638.78    2.98  637.39    5.97  635.54    8.95  633.42   20.89  627.77
   26.86  625.19   29.85  623.29   32.83  622.12    38.8  620.38   45.96617.9978
   47.76  617.45   50.74  617.14   53.73  617.34    60.6617.9976   65.67  618.48
   71.64  619.29   80.45  619.98   83.37  620.74   86.28  621.93   89.19  623.54
   92.11  625.57   97.93  627.97  106.68  632.07  109.59  633.67  115.42  637.49
  121.24  639.96
#Mann= 3 , 0 , 0
       0      .1       0   45.96      .1       0    60.6      .1       0
Bank Sta=45.96,60.6
XS Rating Curve= 0 ,0
Exp/Cntr=0.3,0.1

Type RM Length L Ch R = 1 ,1736.337,100.42,91.11,87.21
XS GIS Cut Line= 2
     613843.9531    4341720.1756     613769.3405    4341635.2442
#Sta/Elev= 28
       0  639.95    6.11   636.3    9.17  635.45   12.22  634.05   18.33  630.25
   21.39  628.09   24.44  625.15   33.61  617.54   36.66  615.33   39.45614.2359
   39.72  614.13   42.78  613.75   45.83  613.79   52.26614.2346   67.22  614.91
   70.27  615.46   73.33  616.49   76.39  618.19   79.44  619.17    82.5   620.3
   91.66  623.93   94.72  625.31   97.77  627.09  100.83  629.23  103.88  632.25
  106.94   635.4  109.99   637.7  113.05  639.89
#Mann= 3 , 0 , 0
       0      .1       0   39.45      .1       0   52.26      .1       0
Bank Sta=39.45,52.26
XS Rating Curve= 0 ,0
Exp/Cntr=0.3,0.1

Type RM Length L Ch R = 1 ,1645.222,51.57,48.59,43.48
XS GIS Cut Line= 4
     613916.1128    4341632.8664     613877.3649    4341620.7026
     613870.1537    4341616.9402     613815.3781    4341582.8566
#Sta/Elev= 30
       0  629.38     2.9  628.88     8.7  627.23    14.5  625.31   17.41  624.08
   20.31  621.68   23.21  620.19   26.11  618.43   31.91  613.78   34.51612.3545
   34.81  612.19   37.71  612.25   40.61  612.89   43.32  612.88   46.03  612.48
   48.75  612.31   64.11  611.64   67.18  611.97   68.66612.3557   70.25  612.77
   82.54  616.43   85.61  617.93   88.68  618.98   94.83  620.37    97.9  621.61
  100.97  623.14  104.04  624.82  107.12  627.58  110.19  629.61  113.26  631.35
#Mann= 3 , 0 , 0
       0      .1       0   34.51      .1       0   68.66      .1       0
Bank Sta=34.51,68.66
XS Rating Curve= 0 ,0
Exp/Cntr=0.3,0.1

Type RM Length L Ch R = 1 ,1596.632,21.35,30.67,32.67
XS GIS Cut Line= 6
     613923.7625    4341632.7634     613922.4396    4341590.0992
     613910.2026    4341576.2086     613895.9812    4341573.5627
     613871.0707    4341572.4118     613828.9489    4341561.4051
#Sta/Elev= 30
       0  628.22   17.14  623.57   19.74  623.05   22.35  622.91   27.56  620.72
   33.29     618   36.16  616.81   38.36   616.1   42.78  615.19   48.07  614.69
   50.71  614.76   53.36  614.59      56  614.17   61.29  613.21   64.18  612.84
   67.08  611.98   69.06611.1579   69.97  610.78   72.86  610.31   84.61  610.37
   93.33611.1573   98.14  612.02  103.69  613.59  106.59  614.66  109.49  616.33
   121.1  619.88  126.91  621.81  132.71  624.96  138.52  626.85  144.32  629.55
#Mann= 3 , 0 , 0
       0      .1       0   69.06      .1       0   93.33      .1       0
Bank Sta=69.06,93.33
XS Rating Curve= 0 ,0
Exp/Cntr=0.3,0.1

Type RM Length L Ch R = 1 ,1565.961,5.89,5.6,5.63
XS GIS Cut Line= 6
     613994.9832    4341726.6351     613962.3124    4341659.2614
     613933.2611    4341591.1576     613914.2111    4341561.9475
      613893.256    4341544.3262     613851.6634    4341529.7212
#Sta/Elev= 30
       0  626.62   17.08  626.63   22.77  626.05    38.1  625.49   50.36  624.66
   53.43  624.39   56.49  623.59   62.62     623   68.75  622.82    77.8  621.71
   89.48  620.71    92.4  620.19   98.24  619.96  124.52  617.16  127.57  617.14
  136.72  616.28  154.74  613.79  169.27  612.51  179.81610.9413   183.8  610.37
  186.73   610.3  204.46610.9415  216.34  611.73  218.73  612.23  234.61  617.12
  237.57  618.16  240.52   619.6  243.47  620.47  252.33  622.32  255.28   623.2
#Mann= 3 , 0 , 0
       0      .1       0  179.81      .1       0  204.46      .1       0
Bank Sta=179.81,204.46
XS Rating Curve= 0 ,0
Exp/Cntr=0.3,0.1

Type RM Length L Ch R = 1 ,1560.361,3.06,3.83,3.89
XS GIS Cut Line= 6
     613943.8753     4341577.057     613931.7045     4341573.882
      613911.896    4341552.5565     613898.4551    4341540.5973
     613892.6475    4341537.8854     613859.3774    4341526.3442
#Sta/Elev= 24
       0  617.98    2.52  617.29    7.55  616.12   12.58  614.58   21.31  613.03
   24.22   612.4   27.13  611.18   29.13610.8157   32.95  610.29   41.68  610.33
   50.68  610.65   53.31610.8166   59.68  611.12   61.81  611.29   63.95  611.55
   67.89  612.44    69.7  612.74   72.74  613.51   75.78  614.43   78.61  614.98
   81.45  615.81   89.97  617.88   95.64  620.27  101.32  621.73
#Mann= 3 , 0 , 0
       0      .1       0   29.13      .1       0   53.31      .1       0
Bank Sta=29.13,53.31
XS Rating Curve= 0 ,0
Exp/Cntr=0.3,0.1

Type RM Length L Ch R = 1 ,1556.531,3.26,2.75,2.99
XS GIS Cut Line= 6
     613944.4433      4341575.01     613938.1991    4341569.8242
     613931.8491    4341566.6492     613898.9349    4341536.6983
     613894.1724    4341534.2773     613863.2875    4341524.4361
#Sta/Elev= 28
       0     618    2.71  617.25   10.48  615.92   12.85  615.47   15.22  614.92
   18.18  614.39   21.15  613.98   24.12  612.78   30.14610.6215   33.02  610.35
   35.98  610.31   38.95  610.33   44.88  610.55   47.85  610.45   50.82  610.53
   56.75  610.27   59.72  610.26    62.4610.6216   65.06  611.06   67.44  611.78
   69.83  612.73    72.9  614.42   75.97  615.45   79.04  615.98   85.19  616.68
   91.34  618.68   94.41  619.94   97.48  620.69
#Mann= 3 , 0 , 0
       0      .1       0   30.14      .1       0    62.4      .1       0
Bank Sta=30.14,62.4
XS Rating Curve= 0 ,0
Exp/Cntr=0.3,0.1

Type RM Length L Ch R = 1 ,1553.782,87.86,91.44,95.51
XS GIS Cut Line= 4
     613953.3926    4341579.9629     613900.4898    4341534.2925
     613895.0075    4341531.7227     613865.0878    4341521.7544
#Sta/Elev= 26
       0  620.45    3.04  619.85    6.08  619.11    9.12  618.48   12.15  617.62
   15.19  616.91   24.31  615.52   33.43  614.23   36.46  612.53    39.5  611.26
   42.54  610.54   45.58  610.34   51.66  610.35   57.73  609.73   59.55609.6282
   66.85  609.15   69.89  609.15   72.39609.6285   75.94   610.5   78.81  611.52
   81.68  613.05   84.54  614.86   87.41  615.43   93.15  617.06  101.75  619.81
  107.48  621.93
#Mann= 3 , 0 , 0
       0      .1       0   59.55      .1       0   72.39      .1       0
Bank Sta=59.55,72.39
XS Rating Curve= 0 ,0
Exp/Cntr=0.3,0.1

Type RM Length L Ch R = 1 ,1462.342,92.5,91.43,91.59
XS GIS Cut Line= 4
     614017.9964    4341526.7648     613977.8334    4341486.7079
     613965.0954    4341478.0137     613937.0337    4341452.9459
#Sta/Elev= 23
       0   631.5    8.96  626.52   11.94  624.46   14.93   621.9    20.9  619.81
   29.85  614.75   32.84  612.99   38.81  608.59    41.8   607.8   51.97606.7657
   64.44  605.91   67.01  606.16   68.86606.7643   69.58     607   72.15  608.35
   83.72  614.85   86.62  616.87   89.51  619.54   92.41   621.2    95.3  622.63
    98.2  623.67  101.09  625.23  109.77   630.4
#Mann= 3 , 0 , 0
       0      .1       0   51.97      .1       0   68.86      .1       0
Bank Sta=51.97,68.86
XS Rating Curve= 0 ,0
Exp/Cntr=0.3,0.1

Type RM Length L Ch R = 1 ,1370.912,42.65,37.57,30.52
XS GIS Cut Line= 3
      614057.684    4341439.4522     614012.1458    4341399.5967
      613978.013    4341380.2561
#Sta/Elev= 24
       0  621.36    3.03  620.12    6.05  619.12    12.1  617.19   21.18  614.48
   27.23  612.02   30.26  611.14   33.28  610.54   36.31  609.52   39.34  608.25
   42.36  606.66   45.19605.4645   45.39  605.38   48.41  604.93   56.79  605.02
   66.55  605.31   68.52605.4666   69.57  605.55   72.59  607.49   81.64   611.7
   90.69  615.71   93.71  618.16   96.73  619.65   99.75  620.96
#Mann= 3 , 0 , 0
       0      .1       0   45.19      .1       0   68.52      .1       0
Bank Sta=45.19,68.52
XS Rating Curve= 0 ,0
Exp/Cntr=0.3,0.1

Type RM Length L Ch R = 1 ,1333.345,26.22,26.09,26.49
XS GIS Cut Line= 6
     614095.7897    4341384.6384     614052.6625    4341374.8488
     614034.4062    4341370.0863     614020.9124    4341368.7634
     614009.7999    4341369.2925     613981.2249    4341366.9113
#Sta/Elev= 22
       0  618.74    5.73  617.31     8.6  616.67   11.47  615.91   14.33  614.65
   20.07  612.71   22.93  611.53   28.87   608.9   35.01  605.77   38.08  605.08
   39.33604.8927   41.15  604.62   44.22   604.4   46.92  604.34   72.17604.8932
   87.78   605.3   90.64  605.75   93.51   607.7  107.85  614.88  110.71  616.51
  113.58  618.75  116.45  620.57
#Mann= 3 , 0 , 0
       0      .1       0   39.33      .1       0   72.17      .1       0
Bank Sta=39.33,72.17
XS Rating Curve= 0 ,0
Exp/Cntr=0.3,0.1

Type RM Length L Ch R = 1 ,1307.253,19.57,27.79,34.79
XS GIS Cut Line= 3
     614084.9417    4341357.9154     614040.7562    4341344.4216
     613984.1353    4341339.3945
#Sta/Elev= 21
       0  613.41    2.89  612.42    5.78   611.3   11.55  608.81   20.21  605.47
   28.87  604.78   34.65  604.21    39.8603.4316   40.43  603.34    46.2  603.12
   55.18  603.22   59.19 603.432   61.16  603.63   73.13   604.2   76.12  604.59
   79.11  606.77    82.1   608.5   94.07  614.79   97.06  616.53  100.05  619.04
  103.04  621.02
#Mann= 3 , 0 , 0
       0      .1       0    39.8      .1       0   59.19      .1       0
Bank Sta=39.8,59.19
XS Rating Curve= 0 ,0
Exp/Cntr=0.3,0.1

Type RM Length L Ch R = 1 ,1279.462,97.85,91.44,70.95
XS GIS Cut Line= 5
     614086.7542    4341338.7134     614048.3562    4341326.2049
     614040.7612    4341318.5797     614021.8863    4341306.5683
     613994.2649    4341304.8213
#Sta/Elev= 20
       0  612.43    2.88  610.85    5.77  608.79    8.65  606.99   11.54  605.96
   14.42  605.54   20.19  604.97   34.61     604   40.38  603.36   45.77  603.02
   51.21602.5244   59.54  601.74   62.33  601.86   65.13  602.45   65.79602.5255
   81.82  604.11   90.12  607.67   95.66  610.14   98.43  611.45   101.2  613.26
#Mann= 3 , 0 , 0
       0      .1       0   51.21      .1       0   65.79      .1       0
Bank Sta=51.21,65.79
XS Rating Curve= 0 ,0
Exp/Cntr=0.3,0.1

Type RM Length L Ch R = 1 ,1188.022,83.63,91.44,108.45
XS GIS Cut Line= 3
     614093.8961    4341246.4506     614033.3915    4341239.0203
     613986.2463    4341242.6018
#Sta/Elev= 23
       0  612.11    3.05  611.56     6.1  611.16   12.19  610.56   15.24  610.15
   27.43  608.97   30.48  608.28   36.58  604.19   39.62  602.79   42.67  601.77
   45.72  601.22   51.82  600.56   57.74598.3235   60.96  597.82   69.82   598.1
   71.52 598.324   72.78  598.49   75.73  599.47   78.69  600.63   90.51  604.63
   93.46  605.79   96.42  607.86  108.24  612.28
#Mann= 3 , 0 , 0
       0      .1       0   57.74      .1       0   71.52      .1       0
Bank Sta=57.74,71.52
XS Rating Curve= 0 ,0
Exp/Cntr=0.3,0.1

Type RM Length L Ch R = 1 ,1096.582,95.71,91.44,83.03
XS GIS Cut Line= 4
     614108.1389    4341208.4563     614080.3507    4341169.5655
     614075.4818    4341158.4998     614053.6094    4341122.7982
#Sta/Elev= 22
       0  603.74    5.97  600.29    8.96  599.16   11.95  598.93   14.94  597.71
   17.92  597.18   20.91  596.91    23.9  596.75   32.86  596.53   35.85  596.36
   38.84  595.29   41.82  593.72   44.18593.4201    47.8  592.74   53.84  593.15
   65.87  593.21   68.86   593.3    70.2 593.421   71.85  593.57   77.83   594.5
   89.79  599.35  101.76  604.08
#Mann= 3 , 0 , 0
       0      .1       0   44.18      .1       0    70.2      .1       0
Bank Sta=44.18,70.2
XS Rating Curve= 0 ,0
Exp/Cntr=0.3,0.1

Type RM Length L Ch R = 1 ,1005.142,95.33,91.44,89.07
XS GIS Cut Line= 2
     614182.9134    4341138.5398      614097.221    4341072.3368
#Sta/Elev= 24
       0  611.92    6.02   608.7   12.03   606.2   15.04  603.47   18.05  601.56
   24.06  598.48   33.09  594.37    36.1  592.32    39.1   589.5    39.4589.4342
   42.11  588.84   54.14  589.27   62.58589.4343   78.21  589.53   81.22  589.73
   84.22  591.11   87.23  592.74   90.24  594.18   93.25  595.54   96.25  596.55
   99.26  598.12  102.27  600.15  105.28  601.97  108.29   604.9
#Mann= 3 , 0 , 0
       0      .1       0    39.4      .1       0   62.58      .1       0
Bank Sta=39.4,62.58
XS Rating Curve= 0 ,0
Exp/Cntr=0.3,0.1

Type RM Length L Ch R = 1 ,913.7023,90.61,91.44,91.51
XS GIS Cut Line= 4
     614243.6691    4341049.8337     614211.4862    4341042.3922
     614195.0428    4341036.2339     614139.3346    4340986.2729
#Sta/Elev= 30
       0  611.95       3  610.24    6.01  608.92    9.01  607.78   12.01  606.37
   15.01  604.62   21.02  600.77   24.02  597.56   27.03  595.23   30.03  593.04
   33.03  590.52   35.96  588.27   36.57588.0435   38.88  587.19   41.81  587.19
   47.66  587.64    57.2588.0449   62.56  588.26   71.54  588.82   74.54  589.45
   83.52  592.76   86.51  593.42    89.5  594.81    92.5  596.67  101.48  600.57
  110.45  604.59  113.45  606.14  116.44   608.3  119.43   609.8  125.42  611.84
#Mann= 3 , 0 , 0
       0      .1       0   36.57      .1       0    57.2      .1       0
Bank Sta=36.57,57.2
XS Rating Curve= 0 ,0
Exp/Cntr=0.3,0.1

Type RM Length L Ch R = 1 ,822.2623,43.12,43.14,43.21
XS GIS Cut Line= 3
     614286.9724    4340975.9541     614249.3903    4340961.1724
     614206.2841    4340933.5649
#Sta/Elev= 22
       0  603.18   11.54  598.27   14.42  597.23   17.31  595.96   20.19   594.3
   34.62  588.34   38.95585.7092   40.38  584.88    43.4  584.56   49.42  584.77
   55.44  585.22   58.45  585.52   59.11585.7086   61.46  586.38   64.47  587.72
   67.48  589.21    70.5  590.38   73.51  591.67   82.54  596.48   85.55  598.93
   88.56  600.67   91.57     602
#Mann= 3 , 0 , 0
       0      .1       0   38.95      .1       0   59.11      .1       0
Bank Sta=38.95,59.11
XS Rating Curve= 0 ,0
Exp/Cntr=0.3,0.1

Type RM Length L Ch R = 1 ,779.1188,45.24,48.3,51.85
XS GIS Cut Line= 2
     614310.3672    4340949.1333     614224.3774    4340893.8353
#Sta/Elev= 16
       0  606.59   18.04  598.22   24.06   595.5   36.08  589.87   39.09  588.34
   43.83585.3328    45.1  584.52   48.11  584.44   54.12  584.92   63.01585.3317
   69.16  586.74   72.17  587.89   84.19   594.6    87.2  596.66   90.21  599.17
  102.24  605.87
#Mann= 3 , 0 , 0
       0      .1       0   43.83      .1       0   63.01      .1       0
Bank Sta=43.83,63.01
XS Rating Curve= 0 ,0
Exp/Cntr=0.3,0.1

Type RM Length L Ch R = 1 ,730.8223,89.46,91.44,93.93
XS GIS Cut Line= 2
     614328.3939    4340919.3099     614266.0587    4340842.8074
#Sta/Elev= 26
       0  603.79    8.97  598.36   14.95  594.59   17.94  593.09   20.93   590.9
   23.92  587.73    29.9   583.6   32.89  582.14   33.32 582.027   35.88  581.35
   38.88  581.65   40.56582.0261   44.86  582.93   47.85  583.42   56.82  584.02
   59.81  584.32    62.8   585.1   65.79  586.32   68.78  587.69   71.77  589.55
   74.76  591.83   77.75  593.47   86.72  598.15   89.71  599.07    92.7  600.17
   98.68  603.18
#Mann= 3 , 0 , 0
       0      .1       0   33.32      .1       0   40.56      .1       0
Bank Sta=33.32,40.56
XS Rating Curve= 0 ,0
Exp/Cntr=0.3,0.1

Type RM Length L Ch R = 1 ,639.3823,91.27,91.44,91.28
XS GIS Cut Line= 2
     614396.0531    4340870.0236     614345.9461    4340775.1781
#Sta/Elev= 23
       0  602.02    3.06  599.97    6.13  599.32    9.19  597.73   15.32  593.68
   21.45   589.5   24.52  586.97   27.58  583.61   30.65   580.6   30.82580.5455
   33.71  579.62   36.78  579.62   42.91  580.39   44.81580.5452    61.3  581.56
   67.43  582.17   70.49  582.72   73.56  584.24   79.68  587.71   95.01  596.08
   98.07  597.97  101.14  598.74  107.27  602.07
#Mann= 3 , 0 , 0
       0      .1       0   30.82      .1       0   44.81      .1       0
Bank Sta=30.82,44.81
XS Rating Curve= 0 ,0
Exp/Cntr=0.3,0.1

Type RM Length L Ch R = 1 ,547.9423,94.04,91.44,84.2
XS GIS Cut Line= 2
     614479.7893    4340832.1381      614421.037    4340725.2558
#Sta/Elev= 30
       0  604.01    3.05  602.33     6.1  600.82    9.15  600.45    12.2  598.94
   24.39   592.2   30.49  587.91   36.59  583.99   39.64  583.04   42.69  581.22
   45.23579.1633   45.74  578.75   48.79  577.75   51.84  578.73   53.96579.1624
   57.93  579.65   60.98  579.81   70.13  579.72   76.23  579.98   79.28  580.55
   82.33  581.54   85.38  582.98   91.47  586.31   94.52  588.09   97.57  590.15
  100.62  591.99  103.67  593.53  106.72  594.03  109.77  595.23  121.97  601.41
#Mann= 3 , 0 , 0
       0      .1       0   45.23      .1       0   53.96      .1       0
Bank Sta=45.23,53.96
XS Rating Curve= 0 ,0
Exp/Cntr=0.3,0.1

Type RM Length L Ch R = 1 ,456.5023,86.55,91.44,90.14
XS GIS Cut Line= 4
      614539.533    4340742.4072     614520.6384    4340728.5736
     614509.5084    4340722.6534     614474.3507    4340689.9919
#Sta/Elev= 25
       0  593.14    2.93  591.09    5.85  588.12    8.78  584.77   11.71  582.17
   14.64  579.77   17.56  578.17   20.41577.8101   28.46   577.9   30.98  577.69
    33.5  577.17   36.02  576.91   39.02  577.06   43.97577.8095   45.02  577.96
   51.02  578.38   54.02  579.07   57.02   580.4   63.02  583.34   66.02  584.29
   69.02  585.36   75.01  588.31   78.01  590.77   81.01  592.65   84.01   594.2
#Mann= 3 , 0 , 0
       0      .1       0   20.41      .1       0   43.97      .1       0
Bank Sta=20.41,43.97
XS Rating Curve= 0 ,0
Exp/Cntr=0.3,0.1

Type RM Length L Ch R = 1 ,365.0623,88.57,91.27,93.6
XS GIS Cut Line= 3
     614613.0207     4340683.255     614558.4013    4340651.5156
     614520.3039    4340620.9178
#Sta/Elev= 22
       0   594.4    6.02  590.65    9.02  588.97   12.03  586.78   15.04  583.99
   21.06  579.67   24.07  577.67   27.07  576.43   30.08  576.07   47.98 575.525
   60.16  575.34   69.28  574.98   72.33  575.04   75.41575.5227    81.5  579.37
   84.55  580.49    87.6  581.47   96.77  586.03   99.82  587.62  102.87  590.06
  105.93  591.76  112.04  594.81
#Mann= 3 , 0 , 0
       0      .1       0   47.98      .1       0   75.41      .1       0
Bank Sta=47.98,75.41
XS Rating Curve= 0 ,0
Exp/Cntr=0.3,0.1

Type RM Length L Ch R = 1 ,273.7893,96.51,91.61,87.3
XS GIS Cut Line= 2
     614655.9081    4340639.9326     614591.7877    4340548.8626
#Sta/Elev= 29
       0  594.66    9.03   590.2   12.04  588.41   15.05  586.35   18.06  584.91
   21.07  584.12   24.08  583.52    30.1  581.34   33.11  580.14   42.14  576.12
   48.16  572.77   50.86571.9178   51.17  571.82   54.18  571.53    60.2  571.54
   66.23   571.7   69.24  571.55   72.43  571.67   75.26  571.89   81.28  571.84
   81.82571.9189   84.29  572.28    87.3  573.03   90.31  573.95   99.34  578.61
  102.35  580.43  105.36  582.66  108.37  584.45  111.38     586
#Mann= 3 , 0 , 0
       0      .1       0   50.86      .1       0   81.82      .1       0
Bank Sta=50.86,81.82
XS Rating Curve= 0 ,0
Exp/Cntr=0.3,0.1

Type RM Length L Ch R = 1 ,182.1824,92.36,91.44,99.64
XS GIS Cut Line= 3
     614732.1083    4340560.5575      614696.112    4340525.1935
     614631.4455     4340488.864
#Sta/Elev= 28
       0  593.62    2.97  592.02    5.94   590.3     8.9  588.97   11.87  588.45
   20.78  583.43   23.75  581.28   26.71  579.55   35.62  574.83   44.52  569.92
   47.49  569.34   50.46  569.24   59.36  568.63   68.26  567.99   69.94567.7693
    74.2  567.33   77.16  567.22   80.13  567.28   88.31567.7688      92  568.14
   94.96  568.62   97.93  569.36   100.9  570.55   109.8  575.34  112.77  577.97
  115.73  580.21   118.7  581.97  124.63  585.64
#Mann= 3 , 0 , 0
       0      .1       0   69.94      .1       0   88.31      .1       0
Bank Sta=69.94,88.31
XS Rating Curve= 0 ,0
Exp/Cntr=0.3,0.1

Type RM Length L Ch R = 1 ,90.74239,26.56,23.04,20.43
XS GIS Cut Line= 6
     614786.2252    4340484.2169     614763.8158    4340461.5834
     614742.8308     4340450.395     614723.1998    4340435.9132
     614720.6886    4340424.0125     614690.0394    4340385.1384
#Sta/Elev= 30
       0  576.39     2.9  575.58    5.79  573.89   14.48  569.64   17.37   568.9
   20.27  568.55   28.96   567.9   31.85  567.72    37.8  567.66   43.74  567.22
   49.69  566.59   52.66  565.78   53.53565.6687   64.78  564.14   67.83  564.08
   73.93  564.52   83.07  564.66   86.11  564.94   92.19  565.12  100.93  564.26
  103.84  564.19  106.75  564.45  112.57  565.36  116.04565.6678   118.4  566.08
  121.31  566.88  127.13  568.77  130.04  569.87  132.96  571.16  141.69  575.79
#Mann= 3 , 0 , 0
       0      .1       0   53.53      .1       0  116.04      .1       0
Bank Sta=53.53,116.04
XS Rating Curve= 0 ,0
Exp/Cntr=0.3,0.1

Type RM Length L Ch R = 1 ,67.69831,17.17,17.9,18.89
XS GIS Cut Line= 5
     614796.3328    4340481.1991     614773.4727    4340436.7491
     614752.6764    4340425.4778     614731.5627     4340418.334
     614702.3526    4340374.8364
#Sta/Elev= 30
       0  577.47    14.7  569.33   17.64  567.95   20.58  567.22   26.46  566.73
    29.4  566.77   38.22  566.13    44.1  565.98   49.98     566   64.77   566.6
   73.64  566.68   76.42  565.95   77.13565.6268   79.21  564.68      82  564.44
   84.78  565.45   87.57  566.11   90.36  566.23   93.14  566.09   98.84  565.23
  107.57   564.6  113.39  564.71   116.3  565.02  119.39565.6276  125.04  566.92
  127.95  567.86  136.68  571.84   142.5  574.95  145.41  576.13  148.32  576.64
#Mann= 3 , 0 , 0
       0      .1       0   77.13      .1       0  119.39      .1       0
Bank Sta=77.13,119.39
XS Rating Curve= 0 ,0
Exp/Cntr=0.3,0.1

Type RM Length L Ch R = 1 ,49.79411,12.46,24.18,33.74
XS GIS Cut Line= 6
     614802.3344     4340475.515     614778.2573    4340423.6566
     614774.6854    4340418.4972     614766.2187    4340412.9409
     614736.9822    4340399.9763     614715.8155    4340369.8138
#Sta/Elev= 30
       0  575.53    3.01  573.93   12.04  568.79   15.05  567.32   18.06  566.43
   21.06  566.01   27.08  565.83   30.09   565.6   35.61565.4566   51.16  565.06
   63.45  565.11   71.05  565.65   79.39   565.9    82.3  565.64   85.21  564.98
   88.11   564.7   91.02  565.43   93.93   565.9   96.84  565.92  105.56  565.29
  108.63  565.27  109.75565.4561   111.7  565.78  117.84  567.12  120.91  567.89
  123.98  568.78  130.13  570.91  136.27  573.37  139.34  573.71  142.41  575.67
#Mann= 3 , 0 , 0
       0      .1       0   35.61      .1       0  109.75      .1       0
Bank Sta=35.61,109.75
XS Rating Curve= 0 ,0
Exp/Cntr=0.3,0.1

Type RM Length L Ch R = 1 ,25.61637,3.68,15.83,18.82
XS GIS Cut Line= 6
     614805.5094    4340473.7952      614779.051    4340413.9993
     614776.1406    4340403.1513     614766.6156    4340389.6575
     614764.7635    4340379.2065     614741.2156    4340354.6002
#Sta/Elev= 28
       0  575.13   11.89  568.52   14.86  567.05   17.83  566.07   20.81  565.66
   23.78  565.71   29.72  565.24   35.67  564.91   41.61  564.83   50.53  564.57
    53.5  564.66   56.47  564.61   71.69564.2429   76.62  564.11   84.88  564.36
   87.63  564.32   94.94   563.9   99.08  563.79  101.42  563.79  103.75  563.91
   105.5564.2427  106.59  564.45  109.43  565.37  112.27  566.39  117.94  568.15
  126.46  571.09  132.13  573.24  137.81  575.56
#Mann= 3 , 0 , 0
       0      .1       0   71.69      .1       0   105.5      .1       0
Bank Sta=71.69,105.5
XS Rating Curve= 0 ,0
Exp/Cntr=0.3,0.1

Type RM Length L Ch R = 1 ,9.790204,6.55,7.41,6.4
XS GIS Cut Line= 6
      614808.705    4340472.7552     614781.5852    4340411.9009
     614779.8654     4340401.053     614784.0987    4340383.0613
     614784.0987    4340377.7696     614747.6817    4340348.6075
#Sta/Elev= 28
       0  575.09    6.06  571.91   12.11  568.44   15.14  566.87   18.17  565.83
    21.2  565.55   24.23  565.43   30.28  564.94    42.4  564.28   54.51  564.34
   66.62  564.14   75.99 563.833   85.53  563.59   93.45  563.97   96.09     564
   98.74  563.83  101.38  563.45   104.3  563.44  107.21  563.72  110.13   563.7
  115.96  563.37  118.88  563.43  121.54563.8322  124.71  564.94  127.62  566.51
  130.54  567.92  136.37  571.27  148.04   575.9
#Mann= 3 , 0 , 0
       0      .1       0   75.99      .1       0  121.54      .1       0
Bank Sta=75.99,121.54
XS Rating Curve= 0 ,0
Exp/Cntr=0.3,0.1

Type RM Length L Ch R = 1 ,2.381145,3.23,2.38,6985.42
XS GIS Cut Line= 6
       614810.91    4340471.9916     614800.7236    4340445.1364
     614786.9652    4340415.1061     614787.0975    4340402.5384
      614791.882    4340381.4599     614750.1439     4340348.916
#Sta/Elev= 30
       0  575.13    8.62  570.48   11.49  568.75   14.36  567.17   17.23  565.91
   20.11  565.52   28.72  564.75   40.73     564   46.74  563.77   58.75  563.94
   65.43563.6853   71.81  563.34   76.69  563.24   83.81  563.38   93.68   563.8
   98.16  563.79  100.36   563.7   103.4  563.33  106.43   563.3  109.46  563.74
   112.5  563.84  115.53  563.55  118.56  563.41   121.6  563.39  124.82563.6838
  127.67  564.64  133.73  567.81  136.77  569.47   139.8  571.54   148.9  575.15
#Mann= 3 , 0 , 0
       0      .1       0   65.43      .1       0  124.82      .1       0
Bank Sta=65.43,124.82
XS Rating Curve= 0 ,0
Exp/Cntr=0.3,0.1

River Reach=Minear Run      ,1
Reach XY= 30
     614791.8493    4340392.8625     614860.5088    4340318.2499
614784.485673688  4340207.897208614776.638240182 4339812.2588788
     614861.6883    4339745.2618     614936.8412    4339494.8649
     615136.8607    4339326.9823     615318.4129    4338730.7414
     615148.8676     4338610.197     614919.2353    4338286.3463
      614670.791     4338293.887     614585.4627    4338184.7461
     614492.5938    4338190.3024     614324.3185    4337944.2394
     614153.6619    4337947.4144     614109.1555    4337861.7661
     614125.8806    4337521.9636     613961.9709     4337383.057
     613909.9801    4337237.4036     613539.2982    4337085.4002
     613498.4199     4336881.406     613316.7094    4336759.2345
     613196.0006     4336565.096     612889.6125    4336454.3677
     612605.8836    4336457.2243     612281.2019    4336267.4392
     612074.4296    4336234.4985     612097.8453    4335917.3947
     612056.5702    4335840.4008     611861.7042    4335777.6944

Type RM Length L Ch R = 1 ,7376.625,3.84,20.21,21.05
XS GIS Cut Line= 5
     614921.8183    4340334.0535      614816.461    4340378.4507
     614809.1585    4340371.4656     614796.4585    4340362.5756
     614750.4209    4340347.5473
#Sta/Elev= 30
       0  574.59    3.01  573.04    6.02  571.61   15.04   567.8   18.05  566.64
   21.06  565.23   24.07  562.56    25.8561.9852   27.08  561.56   42.12  561.61
   45.13  561.48   48.14   560.8   51.15  560.57   54.16  560.73   57.16   561.1
   60.17  561.29   66.19   561.4   84.24  561.23  102.29  561.37  118.49561.9846
  134.77  562.57  139.94  562.86  152.04  563.25  164.15  563.33  167.18  563.98
  170.21  565.31  176.26  568.53  179.29  570.93  182.31  573.16  188.37   575.5
#Mann= 3 , 0 , 0
       0      .1       0    25.8      .1       0  118.49      .1       0
Bank Sta=25.8,118.49
XS Rating Curve= 0 ,0
Exp/Cntr=0.3,0.1

Type RM Length L Ch R = 1 ,7356.419,24.59,41.22,36.09
XS GIS Cut Line= 6
     614921.9307    4340333.2703     614847.3181      4340362.11
     614832.5014     4340366.211     614814.2451    4340349.2776
      614787.919    4340348.8808     614751.5387    4340344.7797
#Sta/Elev= 30
       0  574.89    3.04  573.26    9.11  570.53   21.26  565.54   24.29  562.47
   26.01561.9382   27.33  561.53   30.37  561.45   42.51  561.54   45.55  561.21
   48.58  560.62   51.62  560.62   54.66  560.87   57.69  561.24   60.73  561.42
   74.49  561.27   85.12  561.29   115.6561.9369     132  562.35  134.92  562.52
  137.85  562.81  146.62  563.18  152.72  563.24  158.83  563.01  161.88  563.16
  164.93   564.1  174.08  569.12  177.13   572.9  180.18  574.59  183.23  575.89
#Mann= 3 , 0 , 0
       0      .1       0   26.01      .1       0   115.6      .1       0
Bank Sta=26.01,115.6
XS Rating Curve= 0 ,0
Exp/Cntr=0.3,0.1

Type RM Length L Ch R = 1 ,7315.2  ,115.4,91.44,62.82
XS GIS Cut Line= 6
     614923.7331    4340330.6606     614881.7077    4340341.3124
     614860.1677    4340333.5245     614844.8513    4340325.1005
     614818.2076    4340313.7957     614755.7658    4340310.6207
#Sta/Elev= 30
       0  576.37    2.89  574.61   11.56   570.5   20.23  566.65   23.12  565.07
   26.01  562.71    28.9   561.7   29.37561.6317   31.79  561.28   43.35  561.22
   46.22  560.81   49.08  560.56   51.94  560.68   54.81  560.97   57.67  561.13
   60.53   561.2   96.44561.6317  133.52  562.07   136.5  562.17  139.48  562.44
  142.45  563.34  145.43  564.57  148.41  566.38  151.39  567.32  160.32  569.84
   163.3   570.8  166.27  571.87  169.25  573.81  172.23  575.35   175.2  576.34
#Mann= 3 , 0 , 0
       0      .1       0   29.37      .1       0   96.44      .1       0
Bank Sta=29.37,96.44
XS Rating Curve= 0 ,0
Exp/Cntr=0.3,0.1

Type RM Length L Ch R = 1 ,7223.76 ,28.52,91.44,99.01
XS GIS Cut Line= 6
     614944.8998    4340239.3791     614834.7882      4340234.35
     614821.9166    4340250.4367     614809.1126     4340272.071
     614800.3923    4340280.9168     614754.8839    4340295.2043
#Sta/Elev= 30
       0  576.26   12.25  571.28   15.31  568.96   24.49  565.45   30.62  563.65
   33.68  561.72   36.74  560.51   38.69559.9365    39.8  559.61   42.87  559.45
   45.93  559.54   52.05  559.34   67.36   560.3   70.42  560.28   76.55  559.34
   82.67   559.8   88.79  559.97  110.23  559.57  128.78559.9354   144.8  560.71
  158.45   560.9  171.37  561.45  177.33  561.37  180.31  561.73   183.3  563.71
  186.28  565.35  201.18  570.82  204.16  572.12  207.14  574.07  216.09  576.54
#Mann= 3 , 0 , 0
       0      .1       0   38.69      .1       0  128.78      .1       0
Bank Sta=38.69,128.78
XS Rating Curve= 0 ,0
Exp/Cntr=0.3,0.1

Type RM Length L Ch R = 1 ,7132.32 ,94.7,91.44,84.91
XS GIS Cut Line= 6
     614944.2384    4340226.8114     614821.7178    4340220.4329
     614812.1927    4340216.0673     614775.3633    4340212.6856
     614760.0147    4340196.6551     614714.0504    4340179.1863
#Sta/Elev= 30
       0   576.2     9.2  571.99   12.27  570.15   15.34   569.1    27.6  566.26
   30.67  564.98   33.74  562.59   36.81  560.84   39.87   559.6   42.94  559.38
   46.01  559.45   49.07  559.27   52.14  559.31   61.34  559.91   64.41  559.84
   76.68  559.07   85.88  559.42  130.46558.5621  161.61  558.28  183.53  557.92
  188.31  557.99  190.84558.5604   192.5  559.09  195.58  560.71  198.65  562.83
  214.02  566.94  217.09  568.28  220.16  569.29  235.53  572.89  241.68  575.37
#Mann= 3 , 0 , 0
       0      .1       0  130.46      .1       0  190.84      .1       0
Bank Sta=130.46,190.84
XS Rating Curve= 0 ,0
Exp/Cntr=0.3,0.1

Type RM Length L Ch R = 1 ,7040.88 ,81.12,91.44,80.84
XS GIS Cut Line= 4
     614922.6172    4340132.2182     614827.1536    4340126.7722
     614803.4331    4340124.3014     614764.5141    4340118.7668
#Sta/Elev= 20
       0  568.42    2.99  565.66   14.94  559.31   17.93  558.34   20.92  558.03
   35.86  557.58   41.83  557.31   55.52556.8704   59.76  556.65   62.75  556.61
   77.69  556.65  137.61  556.46  140.63  556.51  143.66  556.76  143.95556.8685
  146.68  557.89  149.71  560.51  152.73  563.44  155.75   565.7  158.78  569.03
#Mann= 3 , 0 , 0
       0      .1       0   55.52      .1       0  143.95      .1       0
Bank Sta=55.52,143.95
XS Rating Curve= 0 ,0
Exp/Cntr=0.3,0.1

Type RM Length L Ch R = 1 ,6949.44 ,92.2,91.44,91.98
XS GIS Cut Line= 6
     614928.9716    4340054.3005     614827.1594    4340051.0485
     614821.5375    4340054.2897     614786.4796    4340054.0251
     614776.3781    4340051.3474     614737.6887    4340060.6328
#Sta/Elev= 30
       0  567.49       3  565.49    8.99  561.06   11.98  559.08   14.98  557.92
   17.98  557.54   53.93  556.27   59.92     556    74.9  555.55   85.28555.0803
   92.88  554.63   95.87  554.62  108.35  554.86  122.96  554.69  134.65  554.66
  143.41  554.77  153.86  555.12  156.92  555.14  159.98  554.75  163.04  554.72
  164.51555.0791  166.11  555.47  172.23  557.74  175.29  558.67  178.35  559.79
  181.41  561.08  184.47  562.25  187.53  563.07  190.59  564.01  193.65  565.13
#Mann= 3 , 0 , 0
       0      .1       0   85.28      .1       0  164.51      .1       0
Bank Sta=85.28,164.51
XS Rating Curve= 0 ,0
Exp/Cntr=0.3,0.1

Type RM Length L Ch R = 1 ,6858    ,97.76,91.42,90.44
XS GIS Cut Line= 4
     614951.9301    4339966.5014     614804.3427    4339960.8563
     614768.9503    4339961.6607     614708.2472    4339965.7377
#Sta/Elev= 30
       0  566.51    9.04   562.2   12.06  559.79   15.07  557.97   18.09  556.67
    21.1  555.77   24.11  555.39   48.23  554.58   54.26   554.3   66.31  553.99
   72.34  553.72   87.41  553.31   93.44  553.06  125.11552.3798  132.62   552.2
   153.6  551.89  168.35  551.85   171.3  551.92  179.21552.3801  189.18  552.57
  192.22  552.71  201.35  552.76  204.39  553.16  207.43  554.07  210.47  555.22
  213.52  556.65  225.68  560.43  228.73  561.47  231.77  563.22  243.94  566.84
#Mann= 3 , 0 , 0
       0      .1       0  125.11      .1       0  179.21      .1       0
Bank Sta=125.11,179.21
XS Rating Curve= 0 ,0
Exp/Cntr=0.3,0.1

Type RM Length L Ch R = 1 ,6766.58 ,38.34,91.46,98.28
XS GIS Cut Line= 3
     614974.9477    4339868.1062     614806.3292    4339863.4347
     614736.0285    4339883.1875
#Sta/Elev= 30
       0  566.49    3.07   563.9    6.13  560.84   15.33  556.48   24.54  552.61
   33.74  551.86   43.84550.3406   52.14  549.08   64.41  547.89   76.67  547.67
   98.14  548.14  134.95  550.51  147.21  551.09  162.55  551.52  174.77   551.6
   183.9  551.39  186.94  551.16  193.02  549.98  198.62  549.74  202.15  549.72
  204.39 550.339  208.24  551.62  214.32  552.78  217.37  553.55  220.41  555.03
  223.45  557.21  226.49  559.92  229.54  563.35  232.58  564.63  241.71  567.21
#Mann= 3 , 0 , 0
       0      .1       0   43.84      .1       0  204.39      .1       0
Bank Sta=43.84,204.39
XS Rating Curve= 0 ,0
Exp/Cntr=0.3,0.1

Type RM Length L Ch R = 1 ,6675.12 ,109.06,91.44,84.63
XS GIS Cut Line= 5
     614974.9477    4339853.8187     614864.4877    4339841.6965
     614841.2438    4339823.9856      614812.361     4339791.971
     614747.9348    4339739.5185
#Sta/Elev= 30
       0  565.76       3  562.96   21.02  553.18   27.03  552.39   42.05  551.05
   55.13550.3194   63.07  549.68    87.1  548.52   96.11  548.71  125.73  550.66
  143.22  551.12  163.34  551.02  171.97  549.89  177.71   550.4   189.4   550.4
  201.27  551.02  204.23   550.9  210.17  549.72  215.37550.3198  219.07  550.67
  222.04  550.38     225  550.44  227.97  551.04  230.94  552.04  239.84  556.23
  242.81  557.87  245.77  560.07  248.74  561.47  260.61  566.02  266.54  567.88
#Mann= 3 , 0 , 0
       0      .1       0   55.13      .1       0  215.37      .1       0
Bank Sta=55.13,215.37
XS Rating Curve= 0 ,0
Exp/Cntr=0.3,0.1

Type RM Length L Ch R = 1 ,6583.68 ,80.25,91.44,68.51
XS GIS Cut Line= 4
     614965.1285    4339754.0368     614885.8765    4339730.7853
     614862.1109    4339721.1446     614791.7432     4339687.558
#Sta/Elev= 30
       0     557    3.06  555.03    6.12  553.61    9.18  552.47   12.24  551.85
   21.41   551.4   36.71  551.02   42.83  550.73   65.72549.9413   96.84  549.01
   99.69  548.98  102.54  549.28  108.24  550.08  111.24  550.39  117.24  550.93
  120.23  551.09  123.23  550.58  126.23   549.8  129.23  550.22  132.23  550.96
  135.23  551.34  138.23  551.36  141.23  551.21  147.23  550.58  153.22  550.27
  162.22   549.5  165.45549.9421  168.22  550.81  183.21  556.67  186.21   558.8
#Mann= 3 , 0 , 0
       0      .1       0   65.72      .1       0  165.45      .1       0
Bank Sta=65.72,165.45
XS Rating Curve= 0 ,0
Exp/Cntr=0.3,0.1

Type RM Length L Ch R = 1 ,6492.24 ,91.03,91.44,89.14
XS GIS Cut Line= 4
     614975.3913    4339682.3137     614945.2024    4339668.7588
     614905.5935    4339672.7197     614811.7473    4339623.7682
#Sta/Elev= 30
       0  557.43    3.01  554.01    6.02  552.21    9.03  550.99   12.03  550.46
   21.06  549.63   27.08  548.88   33.09   548.4    48.4  548.42   54.53  548.06
   57.59  548.03   63.71  548.42   69.84  548.44   81.97  548.08   87.39547.8313
  103.14  547.42  112.21  547.36  121.29  547.45  127.33  547.61  133.38  547.53
  136.62547.8317  139.43  548.39  142.45  548.77  145.48  548.78   148.5  548.92
  151.53  549.54  157.58  551.25  169.67  554.41  175.72  557.09  178.74  558.17
#Mann= 3 , 0 , 0
       0      .1       0   87.39      .1       0  136.62      .1       0
Bank Sta=87.39,136.62
XS Rating Curve= 0 ,0
Exp/Cntr=0.3,0.1

Type RM Length L Ch R = 1 ,6400.8  ,26.4,38.04,41.19
XS GIS Cut Line= 6
     615022.1906    4339616.7443     614956.1175    4339578.5458
     614920.5575    4339579.3598     614901.4602    4339583.0861
     614881.9018    4339582.1177     614846.0246    4339560.8701
#Sta/Elev= 29
       0  558.23    3.05  556.15    6.11  554.51   18.32   549.1   21.37  548.11
   24.42  547.58   33.97546.8818   42.74  546.15   45.79  546.08   88.18  546.57
     103  546.55  120.23  546.83  125.79   546.8  134.14  546.49  136.94  546.46
  139.97546.8818  148.13  548.84  150.93  549.11  153.91   548.8  156.89  548.34
  159.86  548.17  162.84  548.42  165.82   549.2   168.8  550.13  171.78  551.55
  174.76  552.76  183.69  555.52  189.65  557.24  192.63   558.2
#Mann= 3 , 0 , 0
       0      .1       0   33.97      .1       0  139.97      .1       0
Bank Sta=33.97,139.97
XS Rating Curve= 0 ,0
Exp/Cntr=0.3,0.1

Type RM Length L Ch R = 1 ,6362.764,43.91,53.4,54.47
XS GIS Cut Line= 6
     615030.7603    4339604.2333     614931.1444    4339549.8613
     614911.9886    4339545.1517     614903.8923    4339543.5642
     614900.7173    4339541.5005     614860.4609    4339522.9664
#Sta/Elev= 30
       0  559.39    3.07  557.94    6.13  556.29     9.2  553.65   12.27  551.73
   15.34  550.17    18.4  548.77   21.47  547.82   24.54  547.43   35.42546.5239
   39.87  546.04   42.94  545.87   46.01  545.86   58.28  546.13   79.75  546.29
  124.76  546.45  133.21  546.41  135.96  546.29  139.23546.5236  145.25  547.78
  148.21  548.17  151.16  548.01  154.12  548.17  157.07  548.98  160.02  550.55
  162.98  551.64  171.84  554.39  177.75  555.91  180.71  557.05  189.57  558.95
#Mann= 3 , 0 , 0
       0      .1       0   35.42      .1       0  139.23      .1       0
Bank Sta=35.42,139.23
XS Rating Curve= 0 ,0
Exp/Cntr=0.3,0.1

Type RM Length L Ch R = 1 ,6309.36 ,88.47,91.44,92.2
XS GIS Cut Line= 2
     615048.0692    4339572.8479     614894.4643    4339472.6714
#Sta/Elev= 28
       0  558.73    3.06  556.76    6.11  554.23   15.28  549.18   18.34   547.7
   21.39  546.85   27.51   546.3   36.68  545.78   39.73   545.7    48.9  546.02
   58.07  546.03   79.47  545.74   87.95545.5003  116.14  544.32  128.37  543.98
  131.43  543.97  134.48  544.13  137.77  544.74   142.7 545.501  152.82  547.39
  155.88  548.22  158.93  550.09  161.99  551.42  165.05  552.44   168.1   553.3
  174.22  555.29  180.33  556.91  183.38  558.14
#Mann= 3 , 0 , 0
       0      .1       0   87.95      .1       0   142.7      .1       0
Bank Sta=87.95,142.7
XS Rating Curve= 0 ,0
Exp/Cntr=0.3,0.1

Type RM Length L Ch R = 1 ,6217.92 ,79.53,91.44,95.56
XS GIS Cut Line= 4
     615086.9543    4339505.7853     614998.9218    4339433.0556
     614986.3529    4339423.8952     614929.7568    4339375.2703
#Sta/Elev= 30
       0  556.88    9.01   553.4   15.02  551.45   21.03  548.62   30.05  545.64
   36.06  546.18   39.06  546.16   53.21545.0745    60.1  544.62   69.11  544.46
   90.15  544.97  105.17  544.88  108.18  544.68  111.18   544.1  114.19  544.21
  117.45545.0743  121.97  546.18  132.73  547.15  147.65  547.25  150.64  547.38
  153.62   547.9   156.6  549.48  159.59  553.05  162.57  554.29  165.56  554.19
  171.53  553.25  174.51   553.2  183.47  554.49  198.39   556.1  204.36  557.09
#Mann= 3 , 0 , 0
       0      .1       0   53.21      .1       0  117.45      .1       0
Bank Sta=53.21,117.45
XS Rating Curve= 0 ,0
Exp/Cntr=0.3,0.1

Type RM Length L Ch R = 1 ,6126.48 ,96.45,91.44,76.2
XS GIS Cut Line= 6
     615121.3357    4339432.4955     615075.7976    4339405.8167
     615060.4673    4339375.8865     615055.9232    4339360.8342
     615037.2787     4339325.108     614964.6819    4339276.0513
#Sta/Elev= 30
       0  557.61    2.93  554.87     8.8  550.99   14.66  548.24   23.46  543.81
   25.69543.3762   26.39  543.24   29.32  543.19   86.41  542.91   91.65  542.93
   94.27  543.05      97543.3772  102.13  544.07  110.76  544.95   119.4  546.29
  142.43  548.32  151.49  549.54  157.53  549.96  169.62  551.23  172.64  551.46
  175.66  551.49  178.68  552.02   181.7  552.82  184.73  553.37  199.83  554.81
  205.87     555  211.92  555.61  217.96  556.47  227.02  557.53  230.04  558.09
#Mann= 3 , 0 , 0
       0      .1       0   25.69      .1       0      97      .1       0
Bank Sta=25.69,97
XS Rating Curve= 0 ,0
Exp/Cntr=0.3,0.1

Type RM Length L Ch R = 1 ,6035.04 ,92.24,91.44,87.52
XS GIS Cut Line= 4
     615165.4776     4339338.319     615138.5001    4339325.8717
     615127.8799    4339322.2762     614994.7651    4339248.7463
#Sta/Elev= 30
       0  558.74    2.97  557.43    5.94  555.82    8.91  553.79   11.88   551.6
   14.86  548.34   17.83  546.09   23.77  543.29   28.24542.1929   32.51  541.59
   40.92  541.24   47.01  541.18   59.17  541.33   72.52542.1938    83.5  543.15
   95.67  543.95  101.75  544.72  110.88   545.4     120  546.62  123.04  547.71
  126.08  548.25  141.29  550.08  144.33  550.65   156.5  551.21  159.54  551.55
  162.58   552.2  165.62  553.21  168.66  553.77  183.87  555.85     193  558.44
#Mann= 3 , 0 , 0
       0      .1       0   28.24      .1       0   72.52      .1       0
Bank Sta=28.24,72.52
XS Rating Curve= 0 ,0
Exp/Cntr=0.3,0.1

Type RM Length L Ch R = 1 ,5943.6  ,92.43,91.44,86.01
XS GIS Cut Line= 3
     615211.6135    4339253.5264     615157.4438      4339236.69
     615009.8463    4339197.1524
#Sta/Elev= 30
       0  559.18    5.97  557.15    8.96  555.98   11.94  553.78   26.87  547.84
   32.84  543.86   35.83  542.28   37.54541.5283   38.81  540.97    41.8  540.42
   59.78  541.39   65.89  541.39   75.06     541   78.12  540.98   94.55541.5302
   120.9  542.32  123.96  542.64  127.01  543.49  130.07  544.61  133.13  546.25
  136.18  546.87  148.41   548.8  151.46  549.57  154.52  550.11  163.69  551.37
  172.85  552.42  178.97   553.3  191.19  555.39  194.25   556.2  209.53     558
#Mann= 3 , 0 , 0
       0      .1       0   37.54      .1       0   94.55      .1       0
Bank Sta=37.54,94.55
XS Rating Curve= 0 ,0
Exp/Cntr=0.3,0.1
