HEC-RAS study MinearRun.prj: MinearRun

--- MinearRun.g01 (geometry) --- (continued)

Type RM Length L Ch R = 1 ,5852.16 ,82.91,91.44,114.81
XS GIS Cut Line= 3
     615228.1279    4339152.7064     615174.7194    4339150.4809
     615032.8651    4339132.8585
#Sta/Elev= 29
       0  558.71   11.88  553.97   14.85  551.96   17.82  550.14   26.73  545.73
    29.7  544.19   32.67  542.48   35.64  540.51   36.54540.1948   38.61  539.47
   59.54  539.79   80.83  539.95   86.08540.1936   92.99  540.59   96.03  540.88
   108.2  541.42  117.32  541.78  126.45  541.91  129.49  542.08  132.53  542.42
  135.57   543.2  138.61  543.76  153.82  546.12   159.9  548.25  172.07  551.68
  175.11  552.95  178.15  554.03  193.36  557.47   196.4  558.51
#Mann= 3 , 0 , 0
       0      .1       0   36.54      .1       0   86.08      .1       0
Bank Sta=36.54,86.08
XS Rating Curve= 0 ,0
Exp/Cntr=0.3,0.1

Type RM Length L Ch R = 1 ,5760.72 ,99.62,91.44,80.9
XS GIS Cut Line= 5
     615237.8288    4339096.7717     615218.0803    4339074.1021
      615215.064    4339068.0696     615206.4756     4339044.781
     615125.5829    4338992.1703
#Sta/Elev= 30
       0  547.71    3.01  546.23    6.01  545.03   15.03  540.89   18.04  539.94
   21.05  539.47   27.06  538.03   31.15537.2906   37.53  536.37   45.08   535.8
   61.63  536.21   64.65  536.72   73.53537.2915   88.77  538.13    94.8  538.28
  100.83  538.62  106.86  539.28  109.88  539.84  115.91  540.26  124.96  540.59
  127.97  540.82  130.99  541.32     134  541.11  137.02  540.55  140.03  540.31
  143.05  540.38  146.07  541.21  149.08  542.66  155.11  546.74  158.13  548.45
#Mann= 3 , 0 , 0
       0      .1       0   31.15      .1       0   73.53      .1       0
Bank Sta=31.15,73.53
XS Rating Curve= 0 ,0
Exp/Cntr=0.3,0.1

Type RM Length L Ch R = 1 ,5669.28 ,72.58,91.53,100.86
XS GIS Cut Line= 6
     615294.8455     4339004.242     615259.5247    4338981.4241
     615229.7779    4338980.3848     615213.8655    4338983.9209
     615189.1454    4338985.1283     615137.5285    4338949.6964
#Sta/Elev= 30
       0  549.64       3  547.72    6.01   544.5    9.01  542.23   12.01  540.22
   15.02  538.57   18.02  537.69   45.03   537.6      48   537.5   59.73536.6539
   62.89  536.35   68.84  535.52   71.82  535.38   82.68  536.28    89.4536.6545
   93.62  536.86   99.12  536.93  115.85  536.78  124.79  536.87  133.73  537.44
  136.72   537.8  145.66  538.41  148.64   538.8  151.62  539.52   154.6  540.41
  157.59  541.84  160.57  543.07  166.53  544.98  172.49  547.53  175.47  549.08
#Mann= 3 , 0 , 0
       0      .1       0   59.73      .1       0    89.4      .1       0
Bank Sta=59.73,89.4
XS Rating Curve= 0 ,0
Exp/Cntr=0.3,0.1

Type RM Length L Ch R = 1 ,5577.755,95.77,91.36,97.43
XS GIS Cut Line= 3
     615321.8451    4338949.9709     615259.0811    4338908.1415
     615201.9783    4338862.0129
#Sta/Elev= 25
       0  548.13    3.02  546.86    6.03  545.05    9.05  542.11   12.07  540.16
   15.09  538.67    18.1  537.96   39.22  537.23   48.27  537.01   72.41  535.59
   75.48535.3055    84.6  534.44   87.66  534.31  106.01  534.83  108.56 535.305
  109.07   535.4  112.13  536.71  118.25  540.15   121.3  542.24  124.36  543.89
  130.48  545.38   136.6  546.77  139.66  547.41  142.72  547.94  148.83  549.28
#Mann= 3 , 0 , 0
       0      .1       0   75.48      .1       0  108.56      .1       0
Bank Sta=75.48,108.56
XS Rating Curve= 0 ,0
Exp/Cntr=0.3,0.1

Type RM Length L Ch R = 1 ,5486.4  ,92.4,91.44,63.71
XS GIS Cut Line= 4
      615355.437    4338847.1962     615294.2623    4338822.3954
      615246.279    4338794.9765     615190.3366    4338803.8044
#Sta/Elev= 30
       0  549.39       6  546.89       9  545.37      12  543.16      27   537.4
      30     536   33.01   535.2   48.01     535   51.01  534.62   56.59534.1178
   66.01  532.94   69.08  532.88   75.22  533.47   85.33534.1174   90.57  534.51
   93.64  534.82   96.71  535.24  102.85  535.58  108.99  535.76  127.24     536
   133.2  536.15  136.18  536.31  139.16  536.31  142.14   536.2  154.06  535.36
  157.04  535.58  160.03  536.82  168.97  542.89  174.93  546.69  177.91  548.71
#Mann= 3 , 0 , 0
       0      .1       0   56.59      .1       0   85.33      .1       0
Bank Sta=56.59,85.33
XS Rating Curve= 0 ,0
Exp/Cntr=0.3,0.1

Type RM Length L Ch R = 1 ,5394.96 ,94.99,91.54,55.25
XS GIS Cut Line= 4
      615372.377    4338738.9247     615282.8197    4338737.0593
     615247.9183    4338753.3859     615160.9735    4338775.2741
#Sta/Elev= 30
       0  549.01   11.94  547.16   14.93   546.2    20.9  545.14   23.89  544.28
   29.86  542.96   32.84  541.65   35.83  539.87   44.79   535.6   47.77  534.39
   51.68533.0169   53.75  532.11   56.73  531.23   59.72  531.33    62.7  531.79
   67.78533.0164   68.68   533.2   71.66  533.44    95.5  534.51  140.06  535.03
  157.99  535.52  172.94  534.84  178.91  534.37   181.9  533.99  184.89  533.86
  187.88  534.53  202.82  540.07  205.81  542.11  211.79  544.54  217.77  547.25
#Mann= 3 , 0 , 0
       0      .1       0   51.68      .1       0   67.78      .1       0
Bank Sta=51.68,67.78
XS Rating Curve= 0 ,0
Exp/Cntr=0.3,0.1

Type RM Length L Ch R = 1 ,5303.417,97.43,91.34,83.04
XS GIS Cut Line= 4
     615307.8119     4338606.954     615247.3752    4338690.0601
     615220.0047      4338712.64     615147.5875     4338745.745
#Sta/Elev= 30
       0  548.28    3.02  546.68    6.04  545.66    9.07   545.1   12.09  544.86
   18.13  544.99   24.18   543.8    27.2  543.47   30.22  542.55   33.25  542.26
   45.33  542.07   48.36  541.39   57.42   537.8   66.49  535.18   71.34531.9198
   72.54   531.1   75.56  530.17   78.58  530.29   84.46531.9166   87.65  532.34
   96.71  532.82  126.41  533.68  147.43  533.76  181.12  533.04  184.18  533.03
  187.24  533.43   190.3   534.7  202.55  541.67  208.68  546.44  217.87  550.13
#Mann= 3 , 0 , 0
       0      .1       0   71.34      .1       0   84.46      .1       0
Bank Sta=71.34,84.46
XS Rating Curve= 0 ,0
Exp/Cntr=0.3,0.1

Type RM Length L Ch R = 1 ,5212.08 ,69.16,91.44,95.89
XS GIS Cut Line= 6
     615227.0044    4338570.2112     615194.0434    4338596.1824
     615188.0562    4338610.1579     615185.4979    4338632.7384
     615178.5311    4338645.4798     615149.0616    4338673.6292
#Sta/Elev= 30
       0  540.04    5.99   538.7    8.99  537.88   11.99  536.68   14.99  535.11
   20.98  533.23   23.98   532.6   26.98  532.21   35.97  531.53   48.05  531.28
   57.17  529.98   64.89528.4243   68.91  527.52   71.71  527.28   74.52   527.6
   76.98528.4229   80.14  529.78   83.04  530.65   88.85   531.4   97.57  532.93
  100.48  533.04  106.31  532.87  112.13  531.09  115.04  530.89  117.95  531.36
  120.86  532.18  123.77  533.34  129.59  535.91   132.5  537.41  135.41  538.53
#Mann= 3 , 0 , 0
       0      .1       0   64.89      .1       0   76.98      .1       0
Bank Sta=64.89,76.98
XS Rating Curve= 0 ,0
Exp/Cntr=0.3,0.1

Type RM Length L Ch R = 1 ,5120.64 ,95.55,91.44,90.41
XS GIS Cut Line= 4
       615207.27    4338506.0594      615141.465     4338559.754
     615123.7182    4338567.2157     615101.2704    4338577.6697
#Sta/Elev= 25
       0  540.64    3.03  539.14    6.07   537.9     9.1   536.9   15.17  535.71
   21.23  534.67   24.27  534.04    27.3  532.58   30.33   531.3   33.37  530.82
    63.7  530.37   78.87  530.32   87.68  530.52   90.43  530.06   96.84 528.262
  101.43  526.83  104.18  526.18  106.93   526.1  109.69  526.75  111.65 528.261
  112.44  528.87  115.19  532.04  123.44  537.13  126.19  538.63  128.95  539.65
#Mann= 3 , 0 , 0
       0      .1       0   96.84      .1       0  111.65      .1       0
Bank Sta=96.84,111.65
XS Rating Curve= 0 ,0
Exp/Cntr=0.3,0.1

Type RM Length L Ch R = 1 ,5029.2  ,94.29,91.44,94.42
XS GIS Cut Line= 3
     615158.5866    4338405.5175     615085.5629    4338484.2097
     615050.4628     4338513.258
#Sta/Elev= 28
       0  540.76    3.07  539.59    6.13  538.25     9.2  537.48   12.27  536.86
   36.81  533.68   39.87  533.45   42.94  533.04   46.01  532.83   49.08   532.5
   55.21  531.78   64.41  530.55   67.48  530.27   76.68  529.87  107.35  529.15
  110.39  528.84  113.43  528.27  117.56527.2814  122.54  525.81  125.58  525.35
  128.62  526.24  130.02527.2796  131.65  528.49  137.73  533.76  140.77  534.55
   143.8  535.47  146.84  536.57  152.92  539.43
#Mann= 3 , 0 , 0
       0      .1       0  117.56      .1       0  130.02      .1       0
Bank Sta=117.56,130.02
XS Rating Curve= 0 ,0
Exp/Cntr=0.3,0.1

Type RM Length L Ch R = 1 ,4937.76 ,86.62,91.44,90.26
XS GIS Cut Line= 5
     615123.6615    4338357.8924     615028.8228    4338410.5577
     615015.0446    4338429.3462     615005.7744    4338435.3539
     614986.3034    4338458.0169
#Sta/Elev= 30
       0  541.59   12.05  537.77   15.07  537.14   18.08  536.79   27.12  536.51
   30.13  535.98   36.16  534.04   42.19  531.79    45.2  530.89   51.23   530.4
   54.24  529.86   57.25  528.73   63.28  527.53   81.36  526.99  102.45  526.66
  108.48  526.32  111.57525.8761  123.04  523.98  125.95  523.81  128.87  524.19
   134.8525.8778  140.06  527.08  142.83  527.35   148.8  526.61  151.79  526.61
  154.78  527.82  160.75  532.38  166.73  536.07  169.72  539.07   172.7  540.62
#Mann= 3 , 0 , 0
       0      .1       0  111.57      .1       0   134.8      .1       0
Bank Sta=111.57,134.8
XS Rating Curve= 0 ,0
Exp/Cntr=0.3,0.1

Type RM Length L Ch R = 1 ,4846.32 ,92.27,91.45,80.12
XS GIS Cut Line= 5
     615020.9953    4338294.5288     614978.8574    4338343.2589
      614962.855    4338354.3194     614941.3809    4338373.8702
     614914.3917    4338410.5153
#Sta/Elev= 30
       0  539.49    6.14  536.37   12.27  534.73   21.47  530.17   24.54  528.32
   27.61  526.62   30.68  525.69   33.74  525.45   58.29  525.42   61.35  525.22
   62.19525.0339    67.2  523.85   69.98  523.49   72.76  523.58   75.54  524.06
   78.91525.0328    81.1   525.6   83.88  526.12   86.78  526.42   104.2  526.86
  112.92     527  128.09  527.91  131.12  528.01  134.15  527.75  137.19  527.79
  140.22  528.87  146.29  532.75  149.32  533.65  152.36  534.89  158.43  538.91
#Mann= 3 , 0 , 0
       0      .1       0   62.19      .1       0   78.91      .1       0
Bank Sta=62.19,78.91
XS Rating Curve= 0 ,0
Exp/Cntr=0.3,0.1

Type RM Length L Ch R = 1 ,4754.869,96.62,91.43,70.48
XS GIS Cut Line= 3
     614940.3064    4338241.5214     614912.3613    4338279.7506
     614838.9693    4338410.8092
#Sta/Elev= 30
       0  538.52    5.92  535.49   11.84  531.62    14.8  531.07   17.76  529.04
   20.72  527.78   23.68  526.79   26.64   526.1    29.6   525.5   35.52  524.95
   39.21523.9356   41.43  523.01   44.39  522.53   53.48  523.13   58.11523.9337
   74.94  525.72   87.21  526.61   93.34  526.86   105.6  527.95  111.73  528.96
  120.93  530.17  123.99  530.37  127.06  530.33  148.52  531.47  151.58   531.7
  160.78  532.97  166.91  533.46  169.97  534.06  182.24  537.36  197.56  540.98
#Mann= 3 , 0 , 0
       0      .1       0   39.21      .1       0   58.11      .1       0
Bank Sta=39.21,58.11
XS Rating Curve= 0 ,0
Exp/Cntr=0.3,0.1

Type RM Length L Ch R = 1 ,4663.44 ,95.55,91.44,85.47
XS GIS Cut Line= 4
     614824.5015    4338214.8234     614821.9693    4338267.0154
     614826.7978    4338289.2261     614821.2802    4338382.0338
#Sta/Elev= 30
       0  539.74    6.15  534.47   15.37  526.15   18.44  523.89   22.46522.6395
   24.59  522.14   27.66  521.95   46.11   522.5   52.25  522.49   55.09  522.17
   58.14  521.42   60.78  521.18   66.46  521.17    69.3  521.51   73.97522.6382
   77.98  523.46   83.98  523.95   89.98  524.82   98.98  525.82  107.97  526.57
  110.97  526.77  113.97   526.8  125.97   527.7  134.96  528.49  137.96  529.18
  140.96  529.21  143.96  530.21  152.96  533.66  161.96  537.42  167.95  540.09
#Mann= 3 , 0 , 0
       0      .1       0   22.46      .1       0   73.97      .1       0
Bank Sta=22.46,73.97
XS Rating Curve= 0 ,0
Exp/Cntr=0.3,0.1

Type RM Length L Ch R = 1 ,4572    ,61.38,91.44,102.43
XS GIS Cut Line= 4
      614738.429     4338194.635      614724.106    4338249.8684
     614743.9957     4338315.339     614731.1529    4338368.5989
#Sta/Elev= 30
       0  539.43    6.01  537.54    9.01  536.45   12.01  534.67   21.02  527.35
   24.03  525.65   27.03  524.98   30.03  522.97      33521.8513   36.04  521.67
   54.06  521.47   74.91  521.53   86.81  521.45   95.74  521.16   98.71  521.18
  101.69  521.52  103.39 521.852  107.64  522.62  110.61  522.95  116.56  523.19
  125.49  523.98   140.7  524.85  143.75  525.29  146.79  525.42  149.84  526.33
  158.97  530.53  165.05  533.58  174.18   538.7  177.23   539.7  180.27  540.21
#Mann= 3 , 0 , 0
       0      .1       0      33      .1       0  103.39      .1       0
Bank Sta=33,103.39
XS Rating Curve= 0 ,0
Exp/Cntr=0.3,0.1

Type RM Length L Ch R = 1 ,4480.56 ,91.23,91.44,91.97
XS GIS Cut Line= 5
     614708.5631    4338203.6644     614684.1893    4338244.9941
     614664.9274    4338262.0187     614648.6014    4338281.4842
     614621.7744    4338321.4558
#Sta/Elev= 28
       0  530.58       6  524.67       9  522.65      12  521.95   35.99  520.86
   65.12  520.09   70.83  519.87   73.69  519.73   77.44 519.172   82.16  518.19
   84.98  517.96    87.8  518.05   90.63  518.63   92.41519.1722   96.27  520.35
   99.09  521.06   102.1  521.67  105.11  521.88  111.13  521.86  120.16  522.03
  126.17  522.23  129.18  522.41  132.19  523.06   135.2  524.21  138.21   525.6
  141.22   527.4  144.23  529.08  147.23  529.25
#Mann= 3 , 0 , 0
       0      .1       0   77.44      .1       0   92.41      .1       0
Bank Sta=77.44,92.41
XS Rating Curve= 0 ,0
Exp/Cntr=0.3,0.1

Type RM Length L Ch R = 1 ,4389.12 ,106.16,91.44,69.17
XS GIS Cut Line= 3
      614657.112    4338135.9948     614614.6465    4338189.5404
     614544.7799     4338259.407
#Sta/Elev= 30
       0  531.66    5.94  530.22    8.91  529.28   23.77     524   26.74  522.87
   29.71  521.45   32.68  520.54   38.63  520.05   44.57  519.96   65.37  519.12
   68.34  518.86   70.79518.2537   74.33  517.42   77.32  517.11   80.32  517.31
   83.31  517.69   86.31  517.86  101.28  517.71  110.26  518.09  119.24  518.17
   140.2  517.72  143.19  517.89  145.25518.2539  146.19  518.42  149.18  519.48
  152.18  521.12  155.17  523.02  161.16  527.17  164.15  528.95  167.15  531.18
#Mann= 3 , 0 , 0
       0      .1       0   70.79      .1       0  145.25      .1       0
Bank Sta=70.79,145.25
XS Rating Curve= 0 ,0
Exp/Cntr=0.3,0.1

Type RM Length L Ch R = 1 ,4297.68 ,69.98,91.44,103.38
XS GIS Cut Line= 6
      614576.943    4338086.7822     614521.9442    4338168.1876
     614520.2878    4338184.3934     614520.2878    4338197.9533
     614521.9302    4338211.8432     614512.0218    4338232.9594
#Sta/Elev= 30
       0     531    3.07  530.71   15.35  529.21   18.42   528.8   21.49  528.13
   24.56  527.64   27.63  527.32    30.7  526.62   33.77  524.99   36.84  522.94
   39.91  521.79   42.98  521.08   46.05  520.15   52.19  519.28   58.33  518.58
   67.54  517.83   73.68  517.66   95.17  517.44  103.67  517.07     118516.2277
  119.96  515.96  125.38  514.96  128.09  514.97  137.32516.2278  145.08  517.01
  147.99  517.21  150.91  518.86  153.82  520.93  159.66  525.35  165.49  530.15
#Mann= 3 , 0 , 0
       0      .1       0     118      .1       0  137.32      .1       0
Bank Sta=118,137.32
XS Rating Curve= 0 ,0
Exp/Cntr=0.3,0.1

Type RM Length L Ch R = 1 ,4206.24 ,95.53,91.44,86.27
XS GIS Cut Line= 5
      614573.768    4338076.4634     614489.4225    4338127.0669
      614470.619     4338133.554     614457.3508    4338136.6965
     614413.4302    4338150.2823
#Sta/Elev= 30
       0  530.99    3.07  530.46    9.22   528.8   21.52  526.28   27.66  525.22
   33.81  523.09   36.89  522.32   46.11  519.77   49.18  519.56   52.25  519.67
   55.33  519.63   61.48  519.38   92.21  517.81  104.04  517.05  109.73  516.55
  113.19515.9937  115.41  515.47  118.25  514.95  120.98  514.81  138.02  514.81
  144.15  514.99  147.21  515.28  148.73 515.993  150.28  516.72  153.34  519.24
  156.41  520.82  162.54  523.24  168.67  526.18  171.73  528.83  177.86  530.74
#Mann= 3 , 0 , 0
       0      .1       0  113.19      .1       0  148.73      .1       0
Bank Sta=113.19,148.73
XS Rating Curve= 0 ,0
Exp/Cntr=0.3,0.1

Type RM Length L Ch R = 1 ,4114.8  ,90.51,91.36,91.69
XS GIS Cut Line= 4
     614506.3521    4337958.3002     614428.5763    4338051.4575
     614421.8193    4338056.2056     614376.9706    4338100.3818
#Sta/Elev= 30
       0  540.63    6.07  538.12   12.14  535.04   24.27  529.86   27.31  529.42
   30.34  528.52   42.47  523.41   45.51  521.97   48.54  520.26   51.58  518.92
   54.61  518.04   57.64   517.5   63.71  516.98   81.92  517.14   87.98  516.96
  100.12  516.29   111.1515.3311  121.36  514.88  135.61  514.76   147.6  514.27
   150.6  514.71  151.77515.3301   153.6   516.3  159.59  520.85  162.59  522.53
  165.59  523.32  171.58  527.27  174.58  528.97  180.58  532.81  192.57  539.77
#Mann= 3 , 0 , 0
       0      .1       0   111.1      .1       0  151.77      .1       0
Bank Sta=111.1,151.77
XS Rating Curve= 0 ,0
Exp/Cntr=0.3,0.1

Type RM Length L Ch R = 1 ,4023.444,98.18,91.52,84.36
XS GIS Cut Line= 4
      614455.552    4337915.4376     614361.7402    4337988.6239
     614354.1677    4337997.4787     614311.0892     4338071.013
#Sta/Elev= 30
       0  540.26    9.15  537.66   15.25  536.23   18.31  535.23   21.36   534.7
   42.71  529.21   45.76  528.59   61.02  526.37   67.12  524.96   70.17  523.94
   73.22  522.32   82.37  518.89   88.47  517.27   94.58  515.81  100.68  514.46
  104.07513.8976  109.83  512.99  112.86  512.86  127.72  513.22  167.96513.8968
   170.2     514  173.25  515.12  176.29  517.69  179.33  520.54  182.38  522.52
  185.42  524.04  191.51  527.36  203.68  534.26  206.73   534.5  215.86  539.77
#Mann= 3 , 0 , 0
       0      .1       0  104.07      .1       0  167.96      .1       0
Bank Sta=104.07,167.96
XS Rating Curve= 0 ,0
Exp/Cntr=0.3,0.1

Type RM Length L Ch R = 1 ,3931.92 ,89.35,91.44,90.78
XS GIS Cut Line= 5
     614309.9449    4337880.2644     614294.8294    4337916.4766
     614292.2848    4337933.7679     614290.8831     4337956.546
     614267.4328    4338054.3442
#Sta/Elev= 30
       0  541.44    3.02  540.24    6.04  539.36   12.07  536.05   24.15  530.52
   27.17   528.6    33.2  523.55   36.22  521.89   39.24  520.95   45.07   516.6
   47.98  514.94   50.89   513.9   57.05513.0046   62.42  512.69   68.13  512.86
   76.69  512.72   94.78  511.89  100.87  512.11   110.3513.0043  119.16  513.56
   128.3  515.54  131.35   515.8   134.4  516.39  137.44  517.33  140.49  518.59
  143.54  520.14  158.78  528.72  161.82  529.94  164.87  530.69  180.11  540.13
#Mann= 3 , 0 , 0
       0      .1       0   57.05      .1       0   110.3      .1       0
Bank Sta=57.05,110.3
XS Rating Curve= 0 ,0
Exp/Cntr=0.3,0.1

Type RM Length L Ch R = 1 ,3840.48 ,72.98,91.44,95.67
XS GIS Cut Line= 6
     614272.1954    4337845.5875     614206.5054    4337928.6899
     614204.7421     4337950.291     614203.3351     4337953.701
     614202.5728    4337963.2159     614177.7389    4338013.8628
#Sta/Elev= 30
       0  539.84    6.05  539.29   18.16  538.76   24.21   538.3   33.29  537.03
   42.37  535.08    45.4  534.09   54.48  529.86   63.56  525.98   75.66  518.25
   78.69  515.87   81.72  513.96   84.74  512.79    90.8  512.17  105.42511.4903
  116.77  511.17  140.84  511.19  155.68  510.63  158.65  511.06  159.86511.4919
  164.59  513.45  167.56  514.46  170.53  514.74  173.49  516.39  176.46   518.5
  179.43   521.1  188.34  531.08  191.31  534.19  194.28  537.01  197.24  539.56
#Mann= 3 , 0 , 0
       0      .1       0  105.42      .1       0  159.86      .1       0
Bank Sta=105.42,159.86
XS Rating Curve= 0 ,0
Exp/Cntr=0.3,0.1

Type RM Length L Ch R = 1 ,3749.04 ,86.04,91.44,94.07
XS GIS Cut Line= 6
     614272.9891    4337832.0937     614155.9547    4337899.1042
     614141.2637    4337909.7718      614132.744    4337913.3013
     614128.0154    4337914.9781     614097.9767    4337927.7049
#Sta/Elev= 30
       0  540.49    3.07  539.77    6.13  539.41   21.46  537.96   45.98  535.34
   49.04  534.42   55.17  531.37    61.3  528.89   64.37  527.01    70.5  524.37
   73.56  522.32   76.63  519.97   88.89  514.01   91.95  512.82   95.02  512.14
  125.67  510.05  146.96  511.58  149.99  510.96  153.31 509.905  156.09  509.09
  158.63  508.68  162.24   508.5  164.75  508.53  167.26     509  168.86509.9027
  170.22  510.67  176.15  517.91  193.95  533.06  196.91  537.25  199.88  540.65
#Mann= 3 , 0 , 0
       0      .1       0  153.31      .1       0  168.86      .1       0
Bank Sta=153.31,168.86
XS Rating Curve= 0 ,0
Exp/Cntr=0.3,0.1

Type RM Length L Ch R = 1 ,3657.599,90.5,91.36,94.59
XS GIS Cut Line= 3
     614272.1954    4337824.1562     614098.4458    4337827.9838
      614059.643    4337835.3826
#Sta/Elev= 30
       0  540.46    3.05  539.82   15.24   538.1   21.34  536.75   36.59  534.55
   48.78  532.02   54.88  529.93   57.93  528.07   60.98  526.72   76.22  521.48
   85.37   514.1   88.42  512.29   91.47  511.56  106.71   510.7  118.91  510.73
  128.06  510.46  149.26509.1024  158.55   507.2   161.6  506.95  164.64  507.26
  167.69  508.44  168.78509.1002  173.79  512.03  176.83  513.57  179.87  515.86
  182.91  518.78  195.06  525.75   198.1  528.05  201.14  531.89  213.29  539.83
#Mann= 3 , 0 , 0
       0      .1       0  149.26      .1       0  168.78      .1       0
Bank Sta=149.26,168.78
XS Rating Curve= 0 ,0
Exp/Cntr=0.3,0.1

Type RM Length L Ch R = 1 ,3566.236,93,91.52,89.66
XS GIS Cut Line= 4
     614238.2625    4337747.3938     614123.4992    4337740.7792
     614109.2531    4337736.7802     614056.6963    4337732.4563
#Sta/Elev= 30
       0  531.18    12.1  526.11   15.13  523.82   18.15   522.4   27.23  518.82
   33.28  516.17    36.3     514   39.33  512.62   42.35  511.89    48.4  510.95
   57.48  509.99   69.58  509.99   99.83  509.19  114.95  508.93  117.91   508.8
   121.5508.3068  126.79  507.09  129.75  506.88  132.68  506.85  135.61  507.18
  139.17508.3058  147.33  511.03  153.19  513.56  156.12  515.55  159.05  517.73
  170.77  523.46   173.7  525.15  176.63  528.04  179.56  529.55  182.48  531.23
#Mann= 3 , 0 , 0
       0      .1       0   121.5      .1       0  139.17      .1       0
Bank Sta=121.5,139.17
XS Rating Curve= 0 ,0
Exp/Cntr=0.3,0.1

Type RM Length L Ch R = 1 ,3474.72 ,92.02,91.47,86.56
XS GIS Cut Line= 4
     614209.8197    4337649.4978     614099.4425    4337645.6098
     614093.8448    4337647.1259     614028.5798    4337649.4978
#Sta/Elev= 30
       0  531.22    6.14  528.63     9.2   527.5   15.34  525.56   18.41  524.29
   33.75  521.34   36.82  520.53   39.88  518.76   42.95  517.28   46.02  515.23
   49.09  512.74   52.15  510.71   55.22  509.73   58.29  509.31   78.16508.0336
   98.17   506.8  113.35  506.96  116.25  507.24  121.17508.0344  128.12  508.65
  142.96  509.66  145.93  510.18   148.9  511.23  154.84  514.13   157.8  516.22
  160.77  518.59  172.65  524.33  175.62  526.01  178.58  528.58  181.55  530.04
#Mann= 3 , 0 , 0
       0      .1       0   78.16      .1       0  121.17      .1       0
Bank Sta=78.16,121.17
XS Rating Curve= 0 ,0
Exp/Cntr=0.3,0.1

Type RM Length L Ch R = 1 ,3383.253,103.99,91.41,82.06
XS GIS Cut Line= 3
     614180.2001    4337557.6354     614146.9968    4337567.7718
     614001.8744    4337595.4874
#Sta/Elev= 30
       0  531.06    8.68  528.41   11.57  527.42   14.47  526.18   17.36  524.26
   20.25  521.02   23.14  519.26   26.04  517.14   28.93  513.93   31.82  510.28
   34.72  507.72   35.66 507.351   37.73  506.54   40.75   506.1   43.76  505.97
   46.78  506.08   55.82  506.94   82.92507.3492  116.13  507.77  140.25  508.36
  143.26  508.71  146.28  510.04  152.31  514.74  158.34   518.7  161.35  520.52
  164.37  522.19  167.39  524.65   170.4   525.7  173.42  526.92  182.46  530.87
#Mann= 3 , 0 , 0
       0      .1       0   35.66      .1       0   82.92      .1       0
Bank Sta=35.66,82.92
XS Rating Curve= 0 ,0
Exp/Cntr=0.3,0.1

Type RM Length L Ch R = 1 ,3291.84 ,84.87,91.44,95.03
XS GIS Cut Line= 5
     614138.8243    4337450.4601     614102.9741    4337475.0283
     614094.0512    4337497.3354     614084.4002    4337515.7001
     614006.5227    4337570.8022
#Sta/Elev= 30
       0  522.96     2.9  521.87    5.79  519.87    8.69  518.64   11.59  517.66
   14.49  516.56   17.38   515.2   20.28  513.53   28.97  508.13   31.87  506.45
   34.77  505.97   46.46  505.37   49.26505.1375   52.47  504.78   55.47  504.59
   64.48  504.77   67.49  504.64   73.41  504.68   86.19505.1373  100.16  505.64
  106.12  505.76  118.04  506.29  138.91  507.04  159.78  508.02  162.76  508.23
  165.74  509.64  168.73   511.4  174.69  515.72  180.65  519.63  183.63  521.47
#Mann= 3 , 0 , 0
       0      .1       0   49.26      .1       0   86.19      .1       0
Bank Sta=49.26,86.19
XS Rating Curve= 0 ,0
Exp/Cntr=0.3,0.1

Type RM Length L Ch R = 1 ,3200.4  ,83.35,91.44,97.47
XS GIS Cut Line= 4
     614117.9209    4337366.7282     614038.4949    4337428.5197
     614024.8538    4337445.2202     613956.2794    4337502.0087
#Sta/Elev= 30
       0  522.91    9.15  520.57   15.25   518.7    18.3  517.57    24.4  513.85
   30.49  511.21   33.54  510.01   39.64  507.92   42.69  507.03   45.74  506.49
   48.79   506.2   51.84  506.09   97.58  504.97  102.72504.7516  111.41  504.27
  114.11  504.26  125.27  503.43  128.34  503.43  131.41  503.63  137.55  504.16
  140.62  504.61   142.6504.7519  162.11  506.29  177.46   507.8  180.53   508.3
  186.67  510.08  189.74  511.12  192.81  512.41  195.88  514.61  211.23  522.77
#Mann= 3 , 0 , 0
       0      .1       0  102.72      .1       0   142.6      .1       0
Bank Sta=102.72,142.6
XS Rating Curve= 0 ,0
Exp/Cntr=0.3,0.1

Type RM Length L Ch R = 1 ,3108.96 ,96.79,91.44,85.21
XS GIS Cut Line= 5
     614076.0759    4337319.0506     613999.7454    4337370.4528
     613956.5239     4337380.858      613933.852    4337382.7467
     613892.7101    4337408.6718
#Sta/Elev= 30
       0  522.02    18.4  519.03   21.47  518.12   27.61  515.28   30.67  513.61
   33.74  511.67   36.81  508.59   39.88  506.01   42.94  504.97   46.01  504.76
   58.28  504.69   82.82  504.32  104.81503.8511   118.7  503.53  121.66  503.38
  127.59   502.8  139.32  502.97  154.21503.8505  165.31  506.06  171.39  507.03
  174.43  507.38  177.47  508.24  180.51  508.65  189.62   510.2  192.66  511.32
   195.7  512.91  198.74  514.67  201.78   517.4  204.82  519.79  207.86  521.69
#Mann= 3 , 0 , 0
       0      .1       0  104.81      .1       0  154.21      .1       0
Bank Sta=104.81,154.21
XS Rating Curve= 0 ,0
Exp/Cntr=0.3,0.1

Type RM Length L Ch R = 1 ,3017.52 ,93.52,91.45,85.27
XS GIS Cut Line= 4
      614015.527    4337250.5097      613958.745    4337284.1672
     613953.1005    4337289.6485     613843.4706    4337354.6829
#Sta/Elev= 30
       0  522.82       6  520.68       9  519.42      12  517.96      21  512.91
      24  511.51      27  508.82      30   506.6      33  505.31      36  504.28
      39  503.84   48.01  503.28   52.29502.8833   71.25  501.68   73.88   501.7
   79.95  502.08   89.05  502.35  104.23   502.5   119.1502.8831  155.82  503.14
  164.92   503.6  167.96  503.97  174.03  504.21  177.06  505.62   180.1  507.41
  183.13  509.35  186.17  511.44  192.24  515.85  198.31  519.87  201.34  522.15
#Mann= 3 , 0 , 0
       0      .1       0   52.29      .1       0   119.1      .1       0
Bank Sta=52.29,119.1
XS Rating Curve= 0 ,0
Exp/Cntr=0.3,0.1

Type RM Length L Ch R = 1 ,2926.072,93.27,91.42,88.52
XS GIS Cut Line= 4
     613919.6153    4337179.0721        613886.7     4337231.863
     613878.3115    4337254.3353      613823.289    4337333.3205
#Sta/Elev= 29
       0  522.32    2.96  520.57    5.92  520.09   11.85   515.7    23.7  507.29
   26.66   505.1   29.62  503.33   32.59   502.4   38.21502.0062   41.47  501.74
   50.36  501.28   56.29  501.62   59.25  501.65    80.2  501.66   92.21  501.76
   98.23   501.7  137.34   501.7  140.35  501.76     144502.0061  152.38  502.84
  155.39  502.98   161.4  503.47  164.41  505.39  167.42  507.73  170.43  510.18
  173.43  513.02  176.44  516.32  179.45  518.35  182.46  521.28
#Mann= 3 , 0 , 0
       0      .1       0   38.21      .1       0     144      .1       0
Bank Sta=38.21,144
XS Rating Curve= 0 ,0
Exp/Cntr=0.3,0.1

Type RM Length L Ch R = 1 ,2834.653,91.68,91.45,91.35
XS GIS Cut Line= 3
     613820.3964    4337141.3689     613800.5291    4337212.6089
     613768.8025    4337296.8119
#Sta/Elev= 24
       0  523.45    8.88  518.54   17.75  513.78   23.67  510.47   29.58  508.79
    35.5  505.46   41.42  502.41   44.38  501.13   46.57500.6252   47.33  500.45
   53.25  499.99   68.04  499.62   79.96  499.99  111.19500.6248  115.95  500.74
  118.95  501.05  121.95   501.9  124.95  502.14  127.95  503.07  133.95  504.71
  136.95  506.28  157.94  520.32  160.94   521.3  163.94  523.83
#Mann= 3 , 0 , 0
       0      .1       0   46.57      .1       0  111.19      .1       0
Bank Sta=46.57,111.19
XS Rating Curve= 0 ,0
Exp/Cntr=0.3,0.1

Type RM Length L Ch R = 1 ,2743.2  ,89.85,91.44,92.22
XS GIS Cut Line= 5
     613748.9829    4337124.8392     613727.0287    4337154.5809
     613721.5399    4337168.3028     613719.2326    4337172.1932
     613693.3961    4337247.8639
#Sta/Elev= 22
       0  519.91    2.84  516.88    5.69  514.26   17.06  505.72   22.75  501.55
   25.59  500.45   30.18499.5163   31.28  499.28   42.88  498.66   45.83  498.64
   48.79  498.77   65.15  498.99   84.87499.5159   91.81  499.81   94.77  500.08
   97.73  500.13  100.69  500.51  103.65  501.58  106.61  503.39  127.34  517.47
  130.31     518  136.23  522.22
#Mann= 3 , 0 , 0
       0      .1       0   30.18      .1       0   84.87      .1       0
Bank Sta=30.18,84.87
XS Rating Curve= 0 ,0
Exp/Cntr=0.3,0.1

Type RM Length L Ch R = 1 ,2651.76 ,91.72,91.44,92.52
XS GIS Cut Line= 5
     613676.1982    4337051.9395     613641.2464    4337130.2406
     613635.8143    4337138.1078      613634.374    4337144.1626
     613598.5521     4337195.707
#Sta/Elev= 30
       0  522.91    3.06  522.04    9.19  517.71   12.25  515.77   15.31  514.84
   18.37  513.51    24.5  509.33   33.69  502.83   36.75   500.8   39.81  499.07
   42.87  498.32   45.94     498   55.12  497.53   63.33497.5088   79.62  497.03
   95.31  496.83  101.53   496.9  114.47497.5085  116.48  497.69  122.46  498.55
  125.44  498.61  131.42  498.47   137.4  498.86  140.39  499.32  143.38  500.66
  152.35   508.8  155.33  511.81  158.32     515  161.31  519.22   164.3  521.15
#Mann= 3 , 0 , 0
       0      .1       0   63.33      .1       0  114.47      .1       0
Bank Sta=63.33,114.47
XS Rating Curve= 0 ,0
Exp/Cntr=0.3,0.1

Type RM Length L Ch R = 1 ,2560.32 ,84.6,91.27,94.47
XS GIS Cut Line= 3
     613635.0554    4337011.8551     613572.4365    4337069.1013
     613523.4397    4337148.8634
#Sta/Elev= 30
       0  522.35   18.18  512.88   21.21  511.06   24.24  508.75   27.27  506.86
   36.36  501.46   39.39  499.89   42.42  498.89   45.45  498.53   48.48  498.49
   54.54  498.12   57.57  497.81   66.38497.2385   84.84  496.19    93.9  496.12
     109  495.85  118.06  495.89   124.1  496.09  133.16  496.86  142.75497.2381
  151.27  497.68  154.29  498.82  157.31  501.85  160.33  505.67  163.35  509.13
  166.37  511.93  169.39  514.33  172.41   515.2  175.43  517.65  178.45  521.39
#Mann= 3 , 0 , 0
       0      .1       0   66.38      .1       0  142.75      .1       0
Bank Sta=66.38,142.75
XS Rating Curve= 0 ,0
Exp/Cntr=0.3,0.1

Type RM Length L Ch R = 1 ,2469.052,83.95,91.61,95.22
XS GIS Cut Line= 2
     613604.4021    4336975.1159     613463.7373    4337050.8812
#Sta/Elev= 30
       0  522.39    3.07  519.34    9.22     516   18.44  511.19   21.51   509.7
   24.58  507.93   27.65   504.5    33.8  500.44   36.87  498.64   39.94  497.54
   43.02  497.17   63.49 496.627   73.74  496.04   82.96  495.36   86.03  495.24
    89.1  495.53    94.7496.6271  101.39  497.92  107.54  497.98  110.61  498.54
  113.68     500  116.76  501.61   122.9  504.27  125.97  505.88  129.05  507.07
  132.12  508.38  144.41  513.78  147.48  515.46  150.55  517.45  159.77  521.68
#Mann= 3 , 0 , 0
       0      .1       0   63.49      .1       0    94.7      .1       0
Bank Sta=63.49,94.7
XS Rating Curve= 0 ,0
Exp/Cntr=0.3,0.1

Type RM Length L Ch R = 1 ,2377.44 ,95.61,91.44,81.31
XS GIS Cut Line= 5
     613582.9499    4336916.3162      613529.741    4336931.9618
      613497.823    4336930.4048     613469.2847    4336932.2971
     613399.6816     4337004.676
#Sta/Elev= 30
       0  523.62   11.68  517.25    14.6  514.62   17.51  512.31   23.35  508.56
   32.11   502.4   35.03   500.5   37.95  497.76   40.87  496.68   43.79  496.18
   75.12494.5897   84.51   493.7   90.28  493.55   93.14  493.71   97.43  494.59
  101.72  495.57  107.44  496.09  134.28   497.7  149.49  498.98  161.66  500.25
   164.7  500.69  167.75  501.52  173.83   503.7  179.92  505.07  182.96  506.39
     186  508.13  189.05  509.52  204.26  516.16  213.39  519.93  216.43  521.55
#Mann= 3 , 0 , 0
       0      .1       0   75.12      .1       0   97.43      .1       0
Bank Sta=75.12,97.43
XS Rating Curve= 0 ,0
Exp/Cntr=0.3,0.1

Type RM Length L Ch R = 1 ,2286    ,98.93,91.44,89.89
XS GIS Cut Line= 5
     613525.1627    4336830.7656     613473.5592    4336847.4178
     613459.3291    4336860.2926     613447.3066    4336886.8592
     613361.9784    4336988.1396
#Sta/Elev= 30
       0   522.1    6.02  520.79    9.04  519.63   18.07   515.2    24.1  511.93
   27.11  509.92   30.12  507.29    48.2  496.38   51.19493.6582   54.22  492.35
   59.71  492.02   62.45  492.14   65.19  492.53   69.08493.6564   70.67  494.08
   73.41  494.35   96.74  495.72  108.59  496.07  117.62  496.56  132.67  498.01
  147.72  499.04   171.8  501.11  177.82  502.02  183.84  503.63  186.85  504.93
  189.86   505.5  207.92  513.41  225.98  519.93  228.99  519.95  235.01  521.93
#Mann= 3 , 0 , 0
       0      .1       0   51.19      .1       0   69.08      .1       0
Bank Sta=51.19,69.08
XS Rating Curve= 0 ,0
Exp/Cntr=0.3,0.1

Type RM Length L Ch R = 1 ,2194.56 ,92.19,91.46,92.39
XS GIS Cut Line= 4
     613461.9799    4336743.6753     613405.8634     4336776.464
     613389.4451     4336809.932     613333.5356    4336886.2748
#Sta/Elev= 30
       0  513.87    5.91  511.84   14.77  508.18   20.68  504.46    32.5  499.56
   35.45  497.93   38.41   495.7   41.36  493.02   47.27  494.12   53.18  494.55
   76.46  493.63   79.33  493.36   82.31492.7001   87.93  491.46    90.8  491.38
   96.54  491.45  103.99492.6994  108.38  493.41  114.48  495.29  120.59  496.46
  126.69  497.15   132.8  497.47  148.06  499.13  157.22  500.58  169.43  503.16
  172.48  503.43  175.53  504.14  181.64  506.32  187.74  508.98   196.9  513.57
#Mann= 3 , 0 , 0
       0      .1       0   82.31      .1       0  103.99      .1       0
Bank Sta=82.31,103.99
XS Rating Curve= 0 ,0
Exp/Cntr=0.3,0.1

Type RM Length L Ch R = 1 ,2103.102,88.05,91.42,91.62
XS GIS Cut Line= 2
     613448.6296    4336658.7326      613283.657    4336781.8388
#Sta/Elev= 30
       0  514.78    6.14  510.28    9.22  508.89   18.43  509.75   21.51  509.03
   27.65  506.55   36.87  502.27   43.01  498.58   46.08  497.08   49.16  496.12
    55.3  495.53   58.37     495   61.45  494.11   64.52  492.73   67.59   492.4
   73.73  493.87   76.81  494.23  101.39  493.33  150.54  491.92  153.64491.4942
  159.76   490.4  162.83  490.15   165.9  490.12  168.98  490.18  172.05  490.92
  173.41491.4959  181.26  494.92  184.34  496.56  202.77  509.38  205.84  512.21
#Mann= 3 , 0 , 0
       0      .1       0  153.64      .1       0  173.41      .1       0
Bank Sta=153.64,173.41
XS Rating Curve= 0 ,0
Exp/Cntr=0.3,0.1

Type RM Length L Ch R = 1 ,2011.68 ,93.8,91.44,87.18
XS GIS Cut Line= 4
     613373.3202    4336608.2148      613305.879    4336661.2495
     613265.6275    4336681.2831     613231.9904    4336705.9588
#Sta/Elev= 30
       0  511.39   15.32  502.01   18.38  499.76   24.51  496.89   27.58  495.88
   30.64   495.3   36.77  493.05   45.96  491.69   55.15  491.98   64.35  491.86
    76.6  491.28   97.58490.7949  106.78  490.86  112.77  491.18  118.77  491.76
  121.77  491.24  127.76   489.5  130.76  489.06  133.74  488.98  136.72  489.03
   139.7  489.57  143.83490.7957  145.66  491.33  151.62  494.72   154.6  496.78
  157.58  499.36  160.56  501.62  163.54  503.55  166.52  506.41  172.48  512.63
#Mann= 3 , 0 , 0
       0      .1       0   97.58      .1       0  143.83      .1       0
Bank Sta=97.58,143.83
XS Rating Curve= 0 ,0
Exp/Cntr=0.3,0.1

Type RM Length L Ch R = 1 ,1920.24 ,95.65,91.44,74.23
XS GIS Cut Line= 3
     613283.6263    4336543.1271      613230.678    4336596.6696
     613163.2871    4336655.8643
#Sta/Elev= 30
       0  513.81    3.01  512.21    6.02  511.28   12.05  507.15   21.08  501.64
    24.1  499.07   27.11   497.2   30.12  494.52   33.13  492.55   36.14  491.25
   39.16   490.8   45.18  490.46   60.24  491.25   66.27  490.94   70.45489.9313
   72.29  489.32    75.3  488.77   78.29  488.67   84.27  488.75   95.22489.9323
   99.22  490.19  120.15   490.1  123.14  490.25  126.13  491.15  138.09   498.5
  147.06  503.21  150.05  505.25  153.04  505.89  159.02  508.73     165  512.46
#Mann= 3 , 0 , 0
       0      .1       0   70.45      .1       0   95.22      .1       0
Bank Sta=70.45,95.22
XS Rating Curve= 0 ,0
Exp/Cntr=0.3,0.1

Type RM Length L Ch R = 1 ,1828.8  ,90.69,91.4,95.59
XS GIS Cut Line= 5
     613194.0716    4336466.7124     613160.5528    4336520.7148
     613153.9207    4336548.5138     613154.2172    4336553.2578
     613143.1322    4336644.7273
#Sta/Elev= 30
       0  513.42    3.03  511.19    9.08   505.2   15.13  499.32   18.16  496.43
   21.19  493.66   24.21  491.69   27.24  491.01   36.32  490.78   48.43  490.25
   60.53  489.86   83.61489.4553   86.42  489.19   92.14  488.04   94.51  487.82
   127.6  489.02  133.75  489.22  142.96  489.38  143.47489.4547  146.03  489.83
   149.1   491.6  152.17  494.36  155.25   496.9  158.32  498.75  164.46  501.74
  167.53  502.29   170.6  503.27  176.75  506.34  179.82  508.03  189.03  513.52
#Mann= 3 , 0 , 0
       0      .1       0   83.61      .1       0  143.47      .1       0
Bank Sta=83.61,143.47
XS Rating Curve= 0 ,0
Exp/Cntr=0.3,0.1

Type RM Length L Ch R = 1 ,1737.4  ,91.54,91.48,90.36
XS GIS Cut Line= 2
     613123.5667    4336419.7656     613039.9445    4336598.6897
#Sta/Elev= 30
       0  513.62    3.04  511.35    9.12  506.49   12.15  504.15   21.27  497.65
   27.35  493.16   30.38   491.7   33.42  490.98   36.46  489.66    39.5  489.38
   66.85  489.16   94.19  488.75  130.83488.3775  133.69  488.02  136.73  487.79
  139.77  487.36  142.81  487.12  145.85  487.15  148.89  487.38  151.95488.3755
  154.96  489.93     158  491.32  161.04  494.35  164.08  496.74  167.12  498.54
  170.15  499.25  173.19  500.18  191.42  510.15  194.46  512.05   197.5  514.13
#Mann= 3 , 0 , 0
       0      .1       0  130.83      .1       0  151.95      .1       0
Bank Sta=130.83,151.95
XS Rating Curve= 0 ,0
Exp/Cntr=0.3,0.1

Type RM Length L Ch R = 1 ,1645.92 ,92.53,91.44,89.65
XS GIS Cut Line= 4
     613003.5057    4336404.9098     612994.0407    4336479.8764
      612976.033    4336523.3067     612967.9026    4336568.9848
#Sta/Elev= 30
       0  503.13    3.02  500.38    6.04  497.97    9.07  495.77   12.09  494.22
   15.11  493.17   18.13  491.85   24.18  488.92   30.22   487.6   33.23486.2788
   36.27  485.68   39.29  485.66   57.43  486.01   84.38  487.18  102.01  487.51
  104.95  487.42  110.82  486.16  113.76  485.89   116.7   485.9  120.77486.2791
  122.58  486.55  125.48  486.59  128.38  487.09  134.18  487.64  137.08  488.68
  142.88  492.38  151.57  497.32  154.47  498.39  157.37   498.8  168.97  504.64
#Mann= 3 , 0 , 0
       0      .1       0   33.23      .1       0  120.77      .1       0
Bank Sta=33.23,120.77
XS Rating Curve= 0 ,0
Exp/Cntr=0.3,0.1

Type RM Length L Ch R = 1 ,1554.48 ,92.73,91.44,84.57
XS GIS Cut Line= 2
      612914.042    4336422.5608     612872.6653    4336572.5518
#Sta/Elev= 30
       0  504.72    3.05  502.64    9.15  497.35   18.31  489.62   21.36  489.53
   24.41  486.82   26.54485.5001   27.46  484.93   30.51   484.3   33.56  484.23
   48.81   484.6   57.97   484.5   61.02  484.59   64.07  485.01   65.94485.5005
   70.17  486.64   73.22  487.13   76.27   487.2   97.63  486.78  109.83  486.65
  112.88  487.17  115.93  488.17  122.03  488.94  125.08  489.85  128.14  491.33
  140.34  498.09  146.44  501.72  149.49   503.1  152.54  503.37  155.59  505.01
#Mann= 3 , 0 , 0
       0      .1       0   26.54      .1       0   65.94      .1       0
Bank Sta=26.54,65.94
XS Rating Curve= 0 ,0
Exp/Cntr=0.3,0.1

Type RM Length L Ch R = 1 ,1463.04 ,90.84,91.49,92.9
XS GIS Cut Line= 4
     612815.7583    4336399.7577     612813.4928     4336459.228
      612816.828    4336486.3741     612812.0849    4336590.0114
#Sta/Elev= 30
       0  505.35    2.98   504.4   14.88  499.34   17.85     498   20.83  496.28
   23.81  495.66   26.78  494.03   29.76  491.56   32.73   489.4   38.68  485.65
   40.04484.9244   41.66  484.06   44.64   483.2   47.61  483.08   53.56  483.88
   56.54  484.05   59.51  484.53  104.48484.9264  126.53  485.59  135.69  486.82
  141.79  488.13  144.84  488.24  150.94  489.22  153.99  490.08   160.1  492.42
   166.2  495.09   172.3  498.15  175.35  498.33  181.46  500.92  190.61  504.27
#Mann= 3 , 0 , 0
       0      .1       0   40.04      .1       0  104.48      .1       0
Bank Sta=40.04,104.48
XS Rating Curve= 0 ,0
Exp/Cntr=0.3,0.1

Type RM Length L Ch R = 1 ,1371.55 ,91.49,91.39,90.28
XS GIS Cut Line= 3
     612731.6201    4336396.9147     612723.2156    4336436.4938
     612723.4493    4336545.6936
#Sta/Elev= 30
       0  494.67    5.78  492.29    8.67  491.98   11.56  491.08   23.12  486.18
   26.01  485.05    28.9  484.22   31.79  483.89   34.68   483.8   37.57  483.41
   40.46  483.38   42.51482.7169   43.49   482.4   46.53  481.65   49.56   481.5
   52.59  481.62   55.63  482.45   56.28 482.716   58.66  483.69   61.69  484.37
   85.96  483.79   98.09  483.75  107.19  483.84   125.4  484.57  131.46  484.66
   134.5  485.09  137.53  486.55  140.56  488.88  143.59  490.98  149.66  493.78
#Mann= 3 , 0 , 0
       0      .1       0   42.51      .1       0   56.28      .1       0
Bank Sta=42.51,56.28
XS Rating Curve= 0 ,0
Exp/Cntr=0.3,0.1

Type RM Length L Ch R = 1 ,1280.16 ,80.36,91.44,85.6
XS GIS Cut Line= 5
     612665.9023    4336342.6255     612634.7326      4336409.83
     612631.5195    4336444.9571     612633.2234    4336458.8009
      612630.845    4336515.2665
#Sta/Elev= 30
       0  495.81    2.96   494.3    5.93  492.99   11.85  490.95   14.82  490.56
   17.78  489.77   23.71  487.57   26.67  486.69    32.6  485.47   38.52  484.48
   41.49  484.22   53.34  483.91   77.02  482.86   93.96482.3038  100.54  482.07
  109.35  481.07  117.72  480.68   123.3  480.72  138.18  482.21  144.12  482.35
  153.05   482.2  156.41482.3047     159     483  161.97   485.3  164.95   488.3
  167.92  490.73   170.9  491.55  173.87  492.12  176.84  493.54  179.82  495.81
#Mann= 3 , 0 , 0
       0      .1       0   93.96      .1       0  156.41      .1       0
Bank Sta=93.96,156.41
XS Rating Curve= 0 ,0
Exp/Cntr=0.3,0.1

Type RM Length L Ch R = 1 ,1188.72 ,84.88,91.44,94.44
XS GIS Cut Line= 4
     612593.8032    4336298.9691     612558.1833    4336411.8955
     612555.5817    4336436.3941      612542.539    4336465.5789
#Sta/Elev= 29
       0  495.37    3.04  493.64    6.07  493.53    9.11  491.74   12.14  490.34
   15.18  489.41   21.25  487.91    33.4  485.22   39.47   484.5   45.54  483.13
   48.58  482.62   51.61  482.46    75.9  482.13   94.43481.7429  118.41  481.33
  126.62  481.33  137.57  481.16  143.05  480.52  145.95  480.36  148.86  480.38
  151.77  481.17  152.63481.7424  154.67   483.1  157.58  485.46  160.48  486.87
   166.3  489.47   169.2  491.56  172.11  493.54  175.01   496.3
#Mann= 3 , 0 , 0
       0      .1       0   94.43      .1       0  152.63      .1       0
Bank Sta=94.43,152.63
XS Rating Curve= 0 ,0
Exp/Cntr=0.3,0.1

Type RM Length L Ch R = 1 ,1097.28 ,92.16,91.44,91.18
XS GIS Cut Line= 3
     612515.2385    4336284.9095     612479.1378     4336378.445
     612458.8466    4336422.8662
#Sta/Elev= 27
       0  494.79    3.04   493.2    9.11  489.77   12.15  488.17   15.19   486.9
   18.23  485.42   24.31  482.14   27.34  480.81   29.44480.6096   33.42  480.22
   36.46  480.17   78.99  480.59  103.31  480.74  106.36  480.51  109.42   479.9
  112.47  479.45  115.52  479.32  118.57  479.48  121.63  480.27  122.36480.6099
  124.68  481.69  127.73  482.72  130.78  483.99  133.84  484.22  136.89  486.33
  142.99  490.77   149.1   495.1
#Mann= 3 , 0 , 0
       0      .1       0   29.44      .1       0  122.36      .1       0
Bank Sta=29.44,122.36
XS Rating Curve= 0 ,0
Exp/Cntr=0.3,0.1

Type RM Length L Ch R = 1 ,1005.84 ,80.04,91.44,94.77
XS GIS Cut Line= 2
     612423.2977    4336259.4825     612373.6929    4336404.8761
#Sta/Elev= 26
       0  495.49    3.07  493.42    6.14  492.73    9.22  489.69   15.36  483.44
   18.43  480.56   21.51  479.06   23.88478.8824   43.01  478.62    89.1  478.19
   92.17  478.14   98.32  477.86  101.39  477.91  104.46  478.07  107.54  478.47
  108.85478.8839  113.68  480.29  116.75  480.84  119.83   481.6   122.9  482.63
  132.12  486.15  135.19  487.63  138.26  488.46  141.33  489.89  147.48  492.34
  153.62  495.07
#Mann= 3 , 0 , 0
       0      .1       0   23.88      .1       0  108.85      .1       0
Bank Sta=23.88,108.85
XS Rating Curve= 0 ,0
Exp/Cntr=0.3,0.1

Type RM Length L Ch R = 1 ,914.4   ,100.41,91.44,82.71
XS GIS Cut Line= 5
     612348.4553    4336250.1612     612336.5025    4336287.8127
     612324.2421    4336299.5577     612312.6493    4336306.6823
     612247.3306    4336386.0437
#Sta/Elev= 30
       0  494.68    3.04  491.84    6.08  488.69   12.15  481.97   15.19   479.6
   18.23  478.95   24.31  478.62   30.39  478.46   40.94477.9638   45.16  477.75
   50.82  477.33    59.2   476.9   67.37  476.72   70.09  476.91   73.11  477.73
   74.27477.9643   76.13  478.34   79.16  478.74  109.39   480.1  121.48  480.36
   136.6  480.13  139.62  480.27  142.64  480.95  145.67  482.32  148.69  484.04
  151.71  485.52  154.74   487.4  157.76  488.01  160.78  488.99  172.87  494.84
#Mann= 3 , 0 , 0
       0      .1       0   40.94      .1       0   74.27      .1       0
Bank Sta=40.94,74.27
XS Rating Curve= 0 ,0
Exp/Cntr=0.3,0.1

Type RM Length L Ch R = 1 ,822.96  ,79.84,71.11,72.79
XS GIS Cut Line= 4
     612257.6494    4336182.0495      612241.816    4336227.3551
     612243.2875    4336283.1116     612223.5181    4336374.1374
#Sta/Elev= 30
       0  495.19       6  494.17       9  493.83      18  493.21   41.99  493.03
   50.93  492.25   53.86  491.59    56.8  491.37   59.73  490.75   62.67  488.18
   65.61  483.79   68.54  479.81   71.48  477.54   71.83477.4038   74.41   476.4
   77.35  475.92   79.06   475.9   83.22  475.91  105.71477.4028  109.78  477.56
   124.8  478.76  136.82  479.23  157.85  479.69  160.86  480.14  166.87  482.08
  169.87  483.42  172.88  483.67  178.89  487.16  181.89  488.63  196.92  494.97
#Mann= 3 , 0 , 0
       0      .1       0   71.83      .1       0  105.71      .1       0
Bank Sta=71.83,105.71
XS Rating Curve= 0 ,0
Exp/Cntr=0.3,0.1

Type RM Length L Ch R = 1 ,751.8477,9.93,10.2,10.53
XS GIS Cut Line= 6
     612248.1244    4336136.0119     612165.2139     4336179.285
      612164.486    4336235.3074     612168.5077    4336253.9341
     612172.1061    4336256.2625      612178.767    4336333.2894
#Sta/Elev= 30
       0  486.89    6.03  484.37   12.07  483.11   21.12  482.08   24.14  481.54
   27.15  480.54   30.17  479.91   51.29  477.83   72.41  477.85   90.51  477.17
   99.42  476.56  152.45  477.42  161.14  477.11  163.68  476.89  165.99 476.428
  168.17  475.59  170.12  475.11  174.41  474.83  177.64  475.17  181.82476.4297
  183.48  476.88  186.46  476.83  192.43  477.15  213.31  477.48  222.26  478.11
  228.23  478.72   234.2  479.56  240.16  481.27  246.13  482.39   252.1  484.85
#Mann= 3 , 0 , 0
       0      .1       0  165.99      .1       0  181.82      .1       0
Bank Sta=165.99,181.82
XS Rating Curve= 0 ,0
Exp/Cntr=0.3,0.1

Type RM Length L Ch R = 1 ,741.6428,2.46,10.12,9.92
XS GIS Cut Line= 6
     612247.8598    4336126.7515     612164.2513    4336170.1433
     612154.7494    4336232.4499      612158.771    4336251.9233
     612161.7344     4336254.675      612162.581    4336328.1235
#Sta/Elev= 30
       0  487.18    3.04  485.53    9.12  483.67   15.19  482.33   21.27  481.68
   24.31  481.13   27.35   480.2   30.39  479.76   51.66  477.87   75.97  477.34
    97.2  477.19   109.2   476.5  136.22  476.74  145.22  477.08   169.3  477.12
  171.74  477.08  174.18  476.72   175.8476.2245  177.58  475.45  183.31  474.72
  192.42  475.95  198.45476.2236  204.39  476.75  225.35  477.77  231.34  478.24
  234.33  478.94  243.31  481.98  246.31  483.26  252.29  486.42  255.29  486.98
#Mann= 3 , 0 , 0
       0      .1       0   175.8      .1       0  198.45      .1       0
Bank Sta=175.8,198.45
XS Rating Curve= 0 ,0
Exp/Cntr=0.3,0.1

Type RM Length L Ch R = 1 ,731.52  ,37.46,38.89,39.66
XS GIS Cut Line= 6
     612248.9182    4336118.2848      612150.493    4336157.4432
      612152.088    4336231.4889     612152.8394    4336245.1102
     612149.8785    4336270.6404       612133.38    4336307.1677
#Sta/Elev= 30
       0  487.79    3.03  485.95    9.08   484.1   15.13  482.44   18.16  481.74
   27.24  479.96   51.45  477.81   69.61  476.74   84.74  476.54  105.93  476.59
  120.74  476.94  132.59  476.65  156.29  476.59   171.1  476.89  182.72  476.97
  193.63  476.88   196.3476.5252   202.2  474.79  205.06  474.59  210.77  474.91
  216.48  475.44  219.34  475.44  231.59476.5255  239.38  477.14  242.24  477.53
   245.1  478.48  247.96   479.9  250.83  481.12  253.69  481.55  259.42  485.16
#Mann= 3 , 0 , 0
       0      .1       0   196.3      .1       0  231.59      .1       0
Bank Sta=196.3,231.59
XS Rating Curve= 0 ,0
Exp/Cntr=0.3,0.1
